--- BRUSHRN.prj (project) ---

Proj Title=BRUSHRN
Current Plan=p01
Default Exp/Contr=0,0
English Units
Geom File=g01
Geom File=g02
Flow File=f01
Plan File=p01
BEGIN DESCRIPTION:
Stream Name: Brushy Run
Flood Zone: Approximate
Pendleton County, West Virginia
HEC-RAS Version: 5.0.7
Hydrology Method:
Regression equation
END DESCRIPTION:
DSS Export Rating Curves= 0
DSS Export Rating Curve Sorted= 0
DSS Export Volume Flow Curves= 0
DXF OffsetX= 0
DXF OffsetY= 0
DXF ScaleX= 0
DXF ScaleY= 0

--- BRUSHRN.p01 (plan) ---

Plan Title=Floodplain
Program Version=4.00
Geom File=g01
Flow File=f01
K Sum by GR=0
Std Step Tol=0.01
Critical Tol=0.01
Num of Std Step Trials=20
Max Error Tol=0.3
Flow Tol Ratio=0.001
Split Flow NTrial=30
Split Flow Tol=0.02
Split Flow Ratio=0.02
Log Output Level=0
Friction Slope Method=1
Unsteady Friction Slope Method=2
Unsteady Bridges Friction Slope Method=1
Global Log Level=0
CheckData=False
Run HTab=0
Run UNet=0
Run PostProcess=0
UNET Theta=0
UNET Theta Warmup=0
UNET ZTol=0
UNET ZSATol=0
UNET MxIter=0
UNET MaxInSteps=0
UNET DtIC=0
UNET DtMin=0
UNET MaxCRTS=0
UNET WFStab=0
UNET SFStab=0
UNET WFX=0
UNET SFX=0
UNET DSS MLevel=0
UNET DZMax Abort=0
UNET Convert EG Bridges=0
UNET Use Existing IB Tables=0
UNET Froude Limit=0
UNET Froude Power=0
Write IC File=0
Echo Input=False
Echo Output=False
Write Detailed=0

--- BRUSHRN.f01 (steady flow) ---

Flow Title=Flows
Program Version=5.07
Number of Profiles= 6
Profile Names=P100yr,P10yr,P25yr,P50yr,P500yr,P101yr
River Rch & RM=BRUSHRN,Main            ,31916
     561     263     371     464     823     683
River Rch & RM=BRUSHRN,Main            ,29561
     626     293     414     517     918     762
River Rch & RM=BRUSHRN,Main            ,27263
     822     382     542     678    1209    1000
River Rch & RM=BRUSHRN,Main            ,24406
    1007     467     662     829    1484    1225
River Rch & RM=BRUSHRN,Main            ,21164
    1179     546     775     971    1741    1435
River Rch & RM=BRUSHRN,Main            ,17663
    1314     607     863    1081    1942    1599
River Rch & RM=BRUSHRN,Main            ,15263
    1466     676     962    1206    2170    1784
River Rch & RM=BRUSHRN,Main            ,14325
    1657     763    1086    1363    2455    2016
River Rch & RM=BRUSHRN,Main            ,11363
    1846     848    1209    1518    2739    2246
River Rch & RM=BRUSHRN,Main            ,7390
    2187    1003    1430    1797    3252    2662
Boundary for River Rch & Prof#=BRUSHRN,Main            , 1
Up Type= 0
Dn Type= 3
Dn Slope=0.03023
Boundary for River Rch & Prof#=BRUSHRN,Main            , 2
Up Type= 0
Dn Type= 3
Dn Slope=0.03023
Boundary for River Rch & Prof#=BRUSHRN,Main            , 3
Up Type= 0
Dn Type= 3
Dn Slope=0.03023
Boundary for River Rch & Prof#=BRUSHRN,Main            , 4
Up Type= 0
Dn Type= 3
Dn Slope=0.03023
Boundary for River Rch & Prof#=BRUSHRN,Main            , 5
Up Type= 0
Dn Type= 3
Dn Slope=0.03023
Boundary for River Rch & Prof#=BRUSHRN,Main            , 6
Up Type= 0
Dn Type= 3
Dn Slope=0.03023
DSS Import GetInterval= 0
DSS Import GetPeak= 0
DSS Import FillOption= 0

--- BRUSHRN.g01 (geometry) ---

Geom Title=Geometry
Program Version=5.07

River Reach=BRUSHRN         ,Main
Reach XY= 30
2405984.54900001649948.3960000272407095.94300001650620.535999981
2407466.37800002651299.1939999982407384.51635092651835.402743381
2407635.23000002652936.7820000482408599.10700002654220.207000052
2409636.05100001656143.147000042     2410711.691657052.960000035
     2411465.433658344.444000049     2411971.065660076.133000043
2412003.32800001662199.9040000252412792.92200001663743.333999985
     2413500.397664121.9850000422413694.58100001664514.910999974
     2414078.373664765.1150000272414318.18800001665463.431000003
      2414709.55665956.7740000152415162.73700001666223.668000028
     2415673.508666208.624000049     2416435.357 667032.49200002
2417550.56000001667694.158000014     2418273.511667925.113000025
2418532.62700001668651.5799999892418467.53000001669295.547000029
     2418851.902669630.7780000222419360.40499999670718.944000046
2419310.75300002 671696.52300004     2419763.148672926.159000047
     2419697.244673405.1710000052420005.42400002674719.419000045

Type RM Length L Ch R = 1 ,31916   ,300.2,300,299.1
XS GIS Cut Line= 3
     2405741.817      650278.606     2405992.985       649953.76
     2406205.379      649603.412
#Sta/Elev= 30
       0 3357.66    68.9 3335.01   131.1 3312.74   146.3 3309.59   191.8 3295.58
   276.2 3264.26   288.5  3258.3   295.8 3253.38   336.9 3218.43   348.5 3210.51
   358.6 3205.98   387.3 3199.84   403.13190.675   408.2  3189.2   418.1 3189.42
     428 3189.59   444.9 3194.15   472.2 3209.98   491.2 3223.74   502.9 3229.82
   515.9 3234.71   559.6 3261.94     573 3269.03   582.4 3272.23     612 3288.49
   652.5 3308.14   671.2 3315.95   722.7 3334.23   783.8 3361.97   820.3 3376.17
#Mann= 5 ,-1 , 0
       0      .1       0   403.1    .045       0   418.1      .1       0
  604.23      .1       0  742.44      .1       0
Bank Sta=403.1,418.1
XS Rating Curve= 0 ,0
Exp/Cntr=0.3,0.1

Type RM Length L Ch R = 1 ,31616   ,299.7,300,298.3
XS GIS Cut Line= 3
     2406025.835      650432.847     2406244.957      650088.724
 2406449.3006501649735.289720775
#Sta/Elev= 30
       0 3369.91    68.7 3336.51    97.7 3318.79   149.3 3289.96   158.8 3286.31
   182.5 3271.63   215.7 3253.33   294.7 3217.62   348.5 3191.41   361.3 3187.49
   372.9 3185.67   387.4 3173.56   400.53168.078   407.7 3167.23   415.53167.493
   428.6 3168.55   443.5 3172.58   451.7 3176.06   457.5 3181.74   467.5 3188.43
     478 3202.87   480.9 3205.64     521 3230.77   608.8 3271.74     618 3274.53
   651.3 3289.68   681.9  3307.4   747.3 3339.25   758.6 3343.27   816.2 3369.32
#Mann= 6 ,-1 , 0
       0      .1       0   400.5    .045       0   415.5      .1       0
  443.46      .1       0  546.13      .1       0  568.74      .1       0
Bank Sta=400.5,415.5
XS Rating Curve= 0 ,0
Exp/Cntr=0.3,0.1

Type RM Length L Ch R = 1 ,31316   ,299.1,300,299.2
XS GIS Cut Line= 3
     2406312.952      650558.054      2406502.59      650190.976
     2406670.703      649814.639
#Sta/Elev= 30
       0 3337.89    54.1 3310.18    99.8 3288.45   152.1  3258.2   165.6 3253.63
   187.7 3240.61   246.7 3212.31   273.8 3198.21   291.6 3190.58   317.6 3184.43
   352.5 3170.57   369.9 3166.41   395.3 3147.44   399.8 3144.89   405.73144.114
   416.4 3143.23   420.73144.465   426.4 3146.69   435.2 3145.64   449.7  3146.3
   461.5  3151.6   504.2 3184.55   531.5 3212.45   543.6 3220.62   557.8 3232.74
   566.6 3238.83   597.3 3255.97   733.1 3321.93   776.7 3341.41   825.3 3361.38
#Mann= 5 ,-1 , 0
       0      .1       0   405.7    .045       0   420.7      .1       0
  497.38      .1       0  500.82      .1       0
Bank Sta=405.7,420.7
XS Rating Curve= 0 ,0
Exp/Cntr=0.3,0.1

Type RM Length L Ch R = 1 ,31016   ,296.1,300,302.4
XS GIS Cut Line= 3
     2406543.131      650725.508     2406732.101      650363.471
     2406911.253      649958.261
#Sta/Elev= 30
       0  3313.7    63.9 3278.22   114.3 3247.58   135.1  3236.6   176.6 3218.84
   215.1 3199.34   269.2 3180.89   287.2 3173.19   300.8 3170.32   318.9 3163.21
   350.4 3144.84   363.9 3139.62     391 3127.05   400.93125.221   413.4 3124.11
   415.93124.175     423 3125.48   430.9 3128.66   448.4 3129.55   454.5 3131.27
   461.5 3136.27   477.6 3143.81     514 3165.54   568.5 3203.52   601.9 3223.34
   636.4 3240.95     702 3269.83     772 3304.18   824.5 3327.23   851.4 3337.54
#Mann= 3 ,-1 , 0
       0      .1       0   400.9    .045       0   415.9      .1       0
Bank Sta=400.9,415.9
XS Rating Curve= 0 ,0
Exp/Cntr=0.3,0.1

Type RM Length L Ch R = 1 ,30716   ,364.8,366.5,366.3
XS GIS Cut Line= 3
     2406601.975         650774.     2406935.152      650510.628
     2407257.298      650229.531
#Sta/Elev= 30
       0 3297.88    24.4 3289.92    76.8    3256   102.4 3241.56   176.5 3203.37
   235.5 3176.11   269.5 3164.58   301.7 3151.43   313.2 3149.53   338.8 3141.77
   370.1 3124.65   395.7  3112.5   407.1 3108.65   417.23108.389   429.5  3107.2
   432.23107.594   445.4 3109.51   466.9 3117.25   479.1 3124.25   497.9  3137.5
   509.1 3142.53   539.9 3162.51   552.1 3168.46   564.2 3177.61   576.4 3183.12
   583.4 3188.84   600.7 3199.48   637.2 3219.53   815.5  3295.9   852.2 3309.79
#Mann= 3 ,-1 , 0
       0      .1       0   417.2    .045       0   432.2      .1       0
Bank Sta=417.2,432.2
XS Rating Curve= 0 ,0
Exp/Cntr=0.3,0.1

Type RM Length L Ch R = 1 ,30349   ,83.4,83.5,83
XS GIS Cut Line= 2
2406797.32092309650986.1758171072407487.72220885650517.982071061
#Sta/Elev= 30
       0 3275.54     6.6 3269.42    16.2 3257.03    48.6 3235.87     108 3202.15
   170.4 3170.63   209.5 3153.21     224  3148.1   245.3 3141.68   257.9  3139.8
   315.9 3124.11   330.4  3115.4   347.9 3102.15   369.1 3089.16   380.7 3083.89
   396.43081.282   403.7 3081.06   410.83081.855   422.2 3084.09   431.9 3088.55
   449.8 3089.35   467.1 3094.51   504.4 3119.21   527.5 3137.12   547.7 3149.62
   586.5  3170.2   634.8 3192.03   683.2 3210.64     732 3232.35   834.2 3272.72
#Mann= 3 , 0 , 0
       0      .1       0   396.4    .045       0   410.8      .1       0
Bank Sta=396.4,410.8
XS Rating Curve= 0 ,0
Exp/Cntr(USF)=0,0
Exp/Cntr=0.3,0.1

Type RM Length L Ch R = 1 ,30266   ,256.1,259.8,261.8
XS GIS Cut Line= 3
     2406847.193      651056.203     2407191.037      650816.667
     2407518.822      650562.949
#Sta/Elev= 30
       0 3247.83    78.2 3205.45   109.8 3190.92   145.7 3171.19   204.2 3144.38
   228.6 3135.24   272.5  3125.6   291.9 3119.24   306.6  3112.1     331 3097.57
   355.3 3089.92   369.9 3079.72   379.7 3074.93   391.4 3073.43   404.1 3076.27
   415.2 3074.11   428.8 3072.92     435 3074.18   461.2 3072.58   474.3 3075.97
     533 3124.57   554.1 3145.75   576.9 3163.56   619.7 3179.62   676.8 3209.38
   696.9 3216.71   742.2 3228.48   762.3 3235.62   798.1 3255.76   833.6 3269.73
#Mann= 3 , 0 , 0
       0      .1       0   415.2    .045       0     435      .1       0
Bank Sta=415.2,435
XS Rating Curve= 0 ,0
Exp/Cntr=0.3,0.1

Type RM Length L Ch R = 1 ,30006   ,157,180.8,152.8
XS GIS Cut Line= 3
2406885.83325563651147.908394713 2407314.4397605651035.585365469
     2407704.038      650928.131
#Sta/Elev= 30
       0  3241.6    67.1 3204.25   135.9 3169.15     216 3138.42   228.4 3132.48
   240.8 3130.38   296.8 3111.07   315.2 3106.77   335.4 3098.64   348.3 3090.06
   371.8 3067.95   389.6 3054.19   397.9 3049.83   410.3 3049.18   426.9 3051.41
   432.93050.861   447.93050.655   451.7  3051.2   455.8 3053.68   464.1  3067.4
   468.3 3071.29     489 3087.42   502.4 3095.44   596.8 3137.45   671.6 3173.55
   700.7 3185.39     767 3218.99   779.5 3222.26   809.2    3238   847.2 3255.84
#Mann= 3 ,-1 , 0
       0      .1       0   432.9    .045       0   447.9      .1       0
#XS Ineff= 2 , 0
          424.71 3055.08
Permanent Ineff=
       F       F
Bank Sta=432.9,447.9
XS Rating Curve= 0 ,0
Exp/Cntr=0.3,0.1

Type RM Length L Ch R = 1 ,29825   ,231.8,264.3,241.2
XS GIS Cut Line= 3
2406874.41030977 651303.733657612407213.86041162651231.587051177
2407749.33664874651028.870080218
#Sta/Elev= 30
       0 3277.72    24.9 3266.45      29 3260.12    37.1 3243.39    41.2 3239.32
    98.5 3208.54   114.8 3196.67   135.3 3190.37   225.3  3148.5   278.4 3126.29
   290.7 3123.69   348.3 3102.56   388.7 3084.99   394.8 3081.28   407.9  3069.5
   429.2 3044.25   435.2 3040.23   453.7 3039.73   480.6 3036.44   497.7 3037.65
   512.7  3046.7   531.9 3048.68     547 3053.76   581.4 3075.27   620.1 3104.21
   667.8 3132.53   797.1 3199.09   856.9 3232.34   891.2 3249.79   919.6 3261.96
#Mann= 4 ,-1 , 0
       0      .1       0   435.2    .045       0   453.7      .1       0
   460.8      .1       0
#XS Ineff= 2 , 0
                          459.68         3045.25
Permanent Ineff=
       F       F
Bank Sta=435.2,453.7
XS Rating Curve= 0 ,0
Exp/Cntr=0.3,0.1

Type RM Length L Ch R = 1 ,29561   ,401.2,397.1,399.8
XS GIS Cut Line= 4
2406950.69814299651444.2145847092407283.52793476 651337.90154762
2407458.48739471651357.9804436762407888.30104506651420.806210573
#Sta/Elev= 30
       0  3216.3    67.9 3185.02   100.8 3172.28   137.9 3159.62   214.7 3129.17
   226.8  3123.3   239.4 3120.87     315 3094.94   376.8 3077.02   396.9 3069.69
     409 3067.18   443.5 3044.13   473.4 3022.66   477.4 3021.37   497.7 3022.79
   511.1 3021.01   521.7 3019.23   533.6 3020.66   541.9 3030.23   557.9 3042.04
   574.3 3057.08   606.6 3082.16   626.8 3094.72   667.3 3117.44   719.8 3150.46
   780.4 3183.72   816.8 3200.49   869.4 3230.17     926 3257.54   959.9 3275.28
#Mann= 3 ,-1 , 0
       0      .1       0   511.1    .045       0   533.6      .1       0
#XS Ineff= 2 , 0
          495.71 3025.31
Permanent Ineff=
       F       F
Bank Sta=511.1,533.6
XS Rating Curve= 0 ,0
Exp/Cntr=0.3,0.1

Type RM Length L Ch R = 1 ,29164   ,480.7,481,473.3
XS GIS Cut Line= 3
 2406965.6992274651705.5806889012407459.24372268651749.175288648
2407855.47220097651786.671435907
#Sta/Elev= 30
       0 3202.33    77.3 3159.68   117.5 3140.45   149.6 3129.28   193.8 3116.62
   223.6 3105.72   266.1 3088.38     286 3078.45   294.8 3076.52   330.3    3061
   362.5 3049.09   386.5 3035.43   414.7 3012.01   441.2 2995.25   446.8 2993.56
     456 2994.99   478.9 2994.01     495 2997.76     507 2995.64   519.1 2996.63
   523.1  2999.7   531.1 3010.26   551.2 3016.01   567.3 3027.52   612.8 3065.59
   636.1 3078.58   687.4  3112.1   744.1 3144.33   772.2 3162.51   893.5 3229.72
#Mann= 6 ,-1 , 0
       0      .1       0   441.2    .045       0     456      .1       0
   567.3      .1       0  853.39      .1       0  885.08      .1       0
Bank Sta=441.2,456
XS Rating Curve= 0 ,0
Exp/Cntr=0.3,0.1

Type RM Length L Ch R = 1 ,28683   ,368.5,370.1,367.5
XS GIS Cut Line= 3
2407029.74590434 652303.668399622407429.05290434 652213.69139962
2407844.45252171652132.894365008
#Sta/Elev= 30
       0 3103.14      55 3086.22   148.5 3061.56   178.8 3050.22   226.5 3040.75
   242.9 3035.95   265.8 3032.66   275.9 3033.07   320.8 3025.66   332.8  3019.1
   361.8 2998.77   382.4 2985.72     407 2967.71   415.1 2966.17   435.5 2967.74
   455.9 2974.12   484.4 2977.69     495 2983.04   504.8 2989.34   545.5 3023.13
   561.8 3034.63     574 3041.65   590.3 3050.03   624.7 3065.18   667.8  3087.2
     680 3091.91   692.2 3099.07   716.8 3109.93   769.6 3137.17   832.5  3171.9
#Mann= 3 ,-1 , 0
       0      .1       0     407    .045       0   435.5      .1       0
Bank Sta=407,435.5
XS Rating Curve= 0 ,0
Exp/Cntr=0.3,0.1

Type RM Length L Ch R = 1 ,28313   ,358.9,360.1,359.5
XS GIS Cut Line= 3
     2407123.185      652647.138     2407545.082      652547.343
2407946.97946199652432.359875742
#Sta/Elev= 30
       0 3129.99    56.3  3097.4   135.2 3054.37   147.5 3049.02   176.3 3031.58
   188.6 3028.96   217.4 3014.25   287.3  2990.8   303.7  2980.7     316 2969.81
   348.9 2946.29   358.8 2943.65   402.4 2942.62   406.5 2940.95   418.1 2931.63
   422.9  2930.2   435.2 2928.69   443.6 2930.23   454.7 2936.64   468.6 2947.21
   476.9  2955.3   489.4 2972.18   493.5 2976.19   512.9 2990.96   522.6 2999.63
   535.1 3012.98   543.4    3019   656.8 3065.73   805.6 3136.04   851.6 3161.14
#Mann= 3 ,-1 , 0
       0      .1       0   422.9    .045       0   443.6      .1       0
Bank Sta=422.9,443.6
XS Rating Curve= 0 ,0
Exp/Cntr=0.3,0.1

Type RM Length L Ch R = 1 ,27953   ,249.5,239.9,235.7
XS GIS Cut Line= 3
2407192.98055115652993.267850781 2407621.1223304652871.255312776
 2408010.3493304652754.397312776
#Sta/Elev= 30
       0  3092.9    30.9 3082.54   126.6 3057.83   139.1 3051.95   155.7 3050.15
   176.5 3039.59   185.3 3037.11     286 2994.26   330.3 2971.35   351.2 2950.68
     372 2927.22   384.5 2916.65   388.6 2914.35   413.92912.431   438.6 2911.73
   443.6  2911.9   446.9 2912.81   455.2 2920.12   471.9 2919.74   484.5 2924.41
   501.2 2936.39   522.1 2956.93   542.9 2967.55   604.2 2989.57   681.3 3013.62
   751.9 3043.72   785.2 3055.38   797.7 3061.97   826.9 3073.22   851.6 3085.85
#Mann= 3 ,-1 , 0
       0      .1       0   413.9    .045       0   443.6      .1       0
Bank Sta=413.9,443.6
XS Rating Curve= 0 ,0
Exp/Cntr=0.3,0.1

Type RM Length L Ch R = 1 ,27713   ,450.8,450,451.5
XS GIS Cut Line= 3
     2407459.794      653347.064      2407754.03      653058.045
      2408054.11      652780.164
#Sta/Elev= 30
       0 2988.78    23.1 2976.84    45.9 2957.51    57.3  2949.7    68.7 2944.63
    85.9 2940.56   108.7 2936.62   120.1 2939.23   177.2 2935.86   222.9  2942.6
     240 2947.83   273.3 2947.47   308.5 2940.48   319.9 2933.63     336 2920.91
   352.9 2912.26   371.3 2905.89   385.4 2903.95   396.6 2897.93   405.5  2897.4
   429.8 2895.68   437.8 2896.91   446.3 2902.57   481.8 2939.73   491.6 2946.19
   534.8 2967.35   644.4 3011.67   712.4 3043.46   752.6 3064.74   821.4 3095.78
#Mann= 4 ,-1 , 0
       0     .06       0    6.91      .1       0   405.5    .045       0
   437.8      .1       0
Bank Sta=405.5,437.8
XS Rating Curve= 0 ,0
Exp/Cntr=0.3,0.1

Type RM Length L Ch R = 1 ,27263   ,290.2,300,306.7
XS GIS Cut Line= 3
      2407736.95      653718.989     2408010.915       653405.06
     2408300.655      653114.287
#Sta/Elev= 30
       0 3042.07    55.2 3022.17    75.7 3010.37    90.4 3009.23   103.4 3001.66
   124.4 2993.66   142.6 2991.06   252.2 2961.68   288.7 2948.75   308.1 2939.54
   318.9 2931.64     350 2902.68   392.1 2870.71   403.6 2867.36   414.2  2865.1
   422.1 2866.89   429.4 2877.42   433.4 2881.53     452 2887.53   484.4 2905.13
   525.6 2912.44   555.2 2927.59   586.4 2940.94   597.8 2943.03   611.7 2950.86
   647.2 2964.03   678.3 2980.64   752.9 3015.06   785.8 3035.16   827.1 3057.09
#Mann= 4 ,-1 , 0
       0     .06       0  116.33      .1       0   403.6    .045       0
   422.1      .1       0
Bank Sta=403.6,422.1
XS Rating Curve= 0 ,0
Exp/Cntr=0.3,0.1

Type RM Length L Ch R = 1 ,26963   ,303.4,300,296.1
XS GIS Cut Line= 3
2407751.16973342653737.222124258     2408177.123      653631.343
     2408575.732      653543.408
#Sta/Elev= 30
       0 3040.49    65.5 3015.32    77.9 3007.94    90.2 3006.91   102.6  2998.7
   110.8 2997.59   135.6 2985.97   197.4 2949.24   278.9 2908.67   337.5 2866.03
     354  2862.8     387 2862.42   391.1 2860.69   403.5 2860.21   415.9 2858.14
   424.42853.248   436.5 2851.58   452.9 2852.95     457 2856.47   465.2 2875.18
   469.2 2881.83   473.3 2885.43   538.9 2901.02   596.2 2920.03   624.9 2931.52
   633.1 2932.53   668.9 2946.19   682.3 2949.36   780.6 2990.56   847.1 3028.86
#Mann= 4 ,-1 , 0
       0     .06       0  178.34      .1       0   424.4    .045       0
   452.9      .1       0
Bank Sta=424.4,452.9
XS Rating Curve= 0 ,0
Exp/Cntr=0.3,0.1

Type RM Length L Ch R = 1 ,26663   ,303.1,300,293.3
XS GIS Cut Line= 3
     2407905.247      654143.353     2408245.551      653922.121
2408619.12718609653693.645163563
#Sta/Elev= 30
       0 3043.89    52.2 3015.89   125.6 2980.68   134.4 2974.96   151.8 2972.37
   230.8 2936.26   240.3 2930.83   250.1 2928.88   270.3    2918   323.8 2893.78
   348.4 2878.86   362.8 2868.36   382.5 2850.87   394.6 2838.03   403.3 2835.95
   416.7 2837.64     426  2840.8   441.1  2839.8   473.4 2842.57   511.8  2842.4
   519.7  2843.7     548 2859.19   583.7 2872.28   612.8  2884.8   650.6 2905.76
   672.7 2920.85   683.9 2923.85     759 2964.61   801.2 2982.37   843.8 3006.71
#Mann= 5 ,-1 , 0
       0      .1       0   99.08     .06       0  207.64      .1       0
   394.6    .045       0   416.7      .1       0
Bank Sta=394.6,416.7
XS Rating Curve= 0 ,0
Exp/Cntr=0.3,0.1

Type RM Length L Ch R = 1 ,26363   ,293.2,300,307.1
XS GIS Cut Line= 3
     2408207.567      654446.838     2408460.817      654122.323
2408695.81685211653779.032521712
#Sta/Elev= 30
       0 2941.42    13.6 2940.07    55.7 2923.14   115.7 2903.43   244.5 2866.86
     273  2857.9   327.1 2838.51   338.5 2835.98   356.3 2836.49   375.4 2829.89
   389.8 2829.52   397.2 2826.23   409.8 2824.64   429.2 2826.38   435.6 2827.48
   483.7 2826.77   493.4 2829.49   507.6 2838.59   524.8 2851.69   541.8    2861
   556.4 2866.99   580.6 2882.31   617.2  2902.5   654.3 2926.55   671.6 2931.65
   682.4 2939.97   700.4 2950.14   766.6 2982.09   798.7 3002.25   827.7 3016.33
#Mann= 4 ,-1 , 0
       0     .06       0   53.75      .1       0   397.2    .045       0
   429.2      .1       0
Bank Sta=397.2,429.2
XS Rating Curve= 0 ,0
Exp/Cntr=0.3,0.1

Type RM Length L Ch R = 1 ,26063   ,301.5,300,298.3
XS GIS Cut Line= 3
      2408262.18      654510.125      2408656.35      654326.612
2409020.67384055654136.385598243
#Sta/Elev= 30
       0 2930.77       5 2929.51    17.9 2922.03    35.9 2914.02      74 2899.61
   108.2 2888.27   221.2 2855.47   303.9 2822.47   320.4 2818.83   340.4 2816.86
   376.2 2816.18   406.6 2818.29   424.7 2812.29   437.5 2810.37   454.2 2812.35
   473.6 2816.13   503.3 2836.49   555.2 2857.88   604.5 2883.74   643.9 2908.25
   658.6 2913.55   667.6 2921.69   712.1 2943.37   726.9  2953.2   780.4 2982.67
     801 2991.07   818.8 3000.06   825.6 3004.42   839.1 3016.47   845.8 3020.61
#Mann= 4 ,-1 , 0
       0     .06       0   88.83      .1       0   424.7    .045       0
   454.2      .1       0
Bank Sta=424.7,454.2
XS Rating Curve= 0 ,0
Exp/Cntr=0.3,0.1

Type RM Length L Ch R = 1 ,25763   ,365.6,366.8,365.8
XS GIS Cut Line= 3
2408383.71958276654823.080699309     2408728.255      654603.394
     2409098.427      654378.785
#Sta/Elev= 30
       0 2937.49    25.5 2928.58    36.8 2921.96      51 2919.73    74.7 2908.87
   141.7 2884.15     164 2878.73   193.3 2868.12   245.7 2852.94   288.2 2838.92
   302.5 2832.84   335.7 2810.74   352.8 2801.23   361.5 2799.41   383.1 2799.03
   394.7  2796.8   407.9 2794.58   422.4 2797.13     463 2796.87   495.2 2805.94
   517.5 2813.74   541.8 2818.83   570.6 2827.72   626.8 2853.83   687.6 2886.03
   716.5 2903.61   729.7 2907.42     739  2914.6   804.5 2954.39   841.6 2975.13
#Mann= 5 ,-1 , 0
       0      .1       0   27.31     .06       0  135.45      .1       0
   394.7    .045       0   422.4      .1       0
Bank Sta=394.7,422.4
XS Rating Curve= 0 ,0
Exp/Cntr=0.3,0.1

Type RM Length L Ch R = 1 ,25396   ,224.8,233.2,237.7
XS GIS Cut Line= 4
2408504.74976891655064.4320246982408759.02968059655009.434843707
2408926.96305559654896.944724207 2409264.5059853654687.737575343
#Sta/Elev= 30
       0  2924.6    18.4 2916.61    55.2 2914.03    60.2 2911.73    79.8 2897.84
   112.5 2880.43   139.7 2867.43   194.4 2845.12   267.6 2822.01   288.7 2812.69
   303.1 2810.28   358.2 2788.11   394.6 2776.25   414.6 2773.48     430 2768.04
   443.4 2767.48   466.5 2766.29   478.62767.688   504.2 2776.08   532.6 2789.11
   556.2 2802.86   597.3 2821.03   655.4 2850.35   672.8 2860.67   686.4 2865.67
   748.3 2901.07     760 2903.27   774.5 2912.12   815.2 2930.93   859.4 2953.62
#Mann= 5 ,-1 , 0
       0     .06       0  143.07      .1       0   443.4    .045       0
   478.6      .1       0  478.64      .1       0
Bank Sta=443.4,478.6
XS Rating Curve= 0 ,0
Exp/Cntr=0.3,0.1

Type RM Length L Ch R = 1 ,25163   ,159.3,154.5,148.8
XS GIS Cut Line= 3
     2408578.689      655155.475      2408983.54      655109.559
2409404.37723474655057.267408432
#Sta/Elev= 30
       0 2905.14    16.2 2903.27    28.2 2895.68    36.3 2891.62   108.7 2857.16
   165.1 2835.25   205.4 2824.22   217.4 2821.84   229.5  2816.7   245.6 2813.77
   293.9 2791.88   347.7 2772.05   383.8 2756.51   395.6 2752.51   410.7 2750.23
   419.9 2752.29     459  2757.9   467.1 2760.89   480.8 2767.62   559.7 2783.63
   575.9 2789.24   596.8 2792.09   616.2 2798.69   652.5 2807.78   696.9 2821.74
   730.3 2834.51   781.5 2857.64   805.7 2867.32   817.8 2873.85   831.5 2876.41
#Mann= 4 ,-1 , 0
       0     .06       0   84.55      .1       0   395.6    .045       0
   419.9      .1       0
Bank Sta=395.6,419.9
XS Rating Curve= 0 ,0
Exp/Cntr=0.3,0.1

Type RM Length L Ch R = 1 ,25008   ,147.7,145.5,142.7
XS GIS Cut Line= 2
2408744.52875074655430.2841759032409324.46477579655077.050415192
#Sta/Elev= 30
       0 2857.28      12 2851.12      26 2850.59    49.4 2839.62    56.5 2837.46
    68.2 2835.75   114.2 2822.05   126.3 2819.89   213.4 2798.09   278.9 2769.77
   321.1 2753.31   337.2 2744.81   344.5 2741.53   347.5 2741.47   360.32744.756
   367.9 2747.69   377.3  2748.6   386.6 2751.02   400.7 2750.88   414.5 2753.55
     432  2759.4   442.9 2761.73   456.9 2767.75   498.6 2780.97   545.5 2793.13
   569.3 2800.76   583.4 2802.86   606.8 2808.72   634.9 2819.53     679 2841.28
#Mann= 4 ,-1 , 0
       0     .06       0    56.5      .1       0   337.2    .045       0
   360.3      .1       0
Bank Sta=337.2,360.3
XS Rating Curve= 0 ,0
Exp/Cntr(USF)=0,0
Exp/Cntr=0.3,0.1

Type RM Length L Ch R = 1 ,24863   ,452.8,456.6,457.9
XS GIS Cut Line= 3
     2408837.828      655634.655     2409139.935      655354.937
     2409439.033      655075.623
#Sta/Elev= 30
       0 2845.33    28.5 2837.98    52.6  2839.6    93.9 2829.44   105.6 2829.24
   136.3 2823.88   243.9 2801.25   257.5 2793.85   311.8 2769.23   345.8 2756.87
   382.8 2747.66   388.3  2744.3   393.7  2737.5     400  2733.1   413.7 2731.47
   425.1 2732.76     432  2734.1   452.8 2747.09     459 2749.64   467.5 2751.52
   517.3 2769.29   579.8 2786.78     592 2792.35   603.4 2794.87   628.6 2804.44
   700.2 2827.27   745.8 2847.45   793.2 2872.76   807.1 2876.57     821 2883.84
#Mann= 5 ,-1 , 0
       0      .1       0     5.6     .06       0  124.82      .1       0
     400    .045       0   425.1      .1       0
Bank Sta=400,425.1
XS Rating Curve= 0 ,0
Exp/Cntr=0.3,0.1

Type RM Length L Ch R = 1 ,24406   ,144.1,148.4,154
XS GIS Cut Line= 2
2409076.08474245655926.1785703972409763.27915586655483.197595194
#Sta/Elev= 30
       0  2874.4    88.8 2846.38   125.8 2833.05   140.3  2829.5     165 2829.19
   174.5  2827.1   186.6 2820.59   227.1 2805.67   260.2 2791.99   279.2 2782.75
   348.7 2739.51   379.1 2722.55   404.22710.268   417.2  2707.5   429.7 2710.11
   445.8 2716.72   458.6 2719.48     476 2727.88     502 2737.06   526.7 2743.44
   548.3 2751.98   559.8 2754.61   574.5 2766.65   588.5 2772.22   618.8 2788.73
   716.2 2830.72     737 2841.12   750.9 2843.32   759.9 2848.28   817.6 2866.76
#Mann= 6 ,-1 , 0
       0      .1       0   42.97     .06       0  152.97      .1       0
   395.2      .1       0   404.2    .045       0   429.7      .1       0
Bank Sta=404.2,429.7
XS Rating Curve= 0 ,0
Exp/Cntr=0.3,0.1

Type RM Length L Ch R = 1 ,24258   ,298.8,295,289.5
XS GIS Cut Line= 2
     2409081.368      655945.494     2409874.643      655728.158
#Sta/Elev= 30
       0 2880.03     159 2830.31   172.5 2821.38   188.8  2819.7     242 2794.59
   254.4 2790.01   283.5 2775.43     293 2768.75     300 2761.93   309.3  2758.6
   337.4 2739.96     383 2696.67   390.6 2692.33   396.82690.709   403.7 2690.01
   429.22691.647   436.9 2694.13     459 2707.93   470.1 2711.89   481.8 2718.11
   590.4 2753.59   606.9 2760.72   618.5 2763.45   628.3 2769.02   660.8 2783.09
   743.8 2808.95   784.6 2823.75   794.3 2828.77     806 2831.11   822.5 2838.32
#Mann= 6 ,-1 , 0
       0      .1       0      66     .06       0  212.78      .1       0
   396.8    .045       0   429.2      .1       0   429.3      .1       0
Bank Sta=396.8,429.2
XS Rating Curve= 0 ,0
Exp/Cntr=0.3,0.1

Type RM Length L Ch R = 1 ,23963   ,407.5,406.7,406.9
XS GIS Cut Line= 3
     2409268.028       656329.01     2409606.824      656099.924
      2409948.49       655868.87
#Sta/Elev= 30
       0 2875.41   104.7 2822.16   181.2 2789.52   191.6 2781.57   206.1 2779.58
   225.2 2772.71   233.9 2767.55   302.7 2737.59   317.1 2728.32   326.8 2726.34
   360.6 2702.63   396.5 2669.96   408.9 2668.11   418.5 2669.94     433 2676.08
   476.5 2684.81   500.6 2694.57   513.4 2698.11   568.1  2719.5     620 2742.55
   640.7 2753.13   664.8 2763.34   674.5 2765.62   683.3 2770.79   703.4 2779.13
   722.8 2786.01   781.3 2802.61   804.3 2813.15   814.5 2814.21   821.4  2816.8
#Mann= 5 ,-1 , 0
       0      .1       0  206.89     .06       0  316.35      .1       0
   396.5    .045       0   418.5      .1       0
Bank Sta=396.5,418.5
XS Rating Curve= 0 ,0
Exp/Cntr=0.3,0.1

Type RM Length L Ch R = 1 ,23556   ,191.2,193.3,188.7
XS GIS Cut Line= 2
2409577.10981196656639.3598119582410220.15441529656115.141601385
#Sta/Elev= 30
       0 2866.58    13.4 2858.85    44.1 2837.58   193.1 2757.17     209 2747.93
   220.4 2738.32     235 2735.41     273 2712.89   285.8 2708.93   322.1 2690.86
   331.3 2684.13   359.7 2657.36   368.5 2650.48   378.8 2646.47   389.2 2647.07
   399.5 2646.25   420.1  2647.3   436.5 2651.85   464.9 2649.35   476.3 2650.18
   494.5  2656.3   533.7 2680.91   570.1 2706.38   583.2  2711.5   598.5 2722.57
     673 2764.19   763.4 2802.49   774.8 2804.91   791.7 2813.99   829.6 2829.23
#Mann= 5 ,-1 , 0
       0      .1       0  172.69     .06       0   365.7      .1       0
   389.2    .045       0   420.1      .1       0
#XS Ineff= 2 , 0
                          438.23         2658.63
Permanent Ineff=
       F       F
Bank Sta=389.2,420.1
XS Rating Curve= 0 ,0
Exp/Cntr=0.3,0.1

Type RM Length L Ch R = 1 ,23363   ,154.6,150,146.6
XS GIS Cut Line= 3
2409721.44384271656792.745685424     2410025.753      656507.812
     2410321.387      656210.556
#Sta/Elev= 30
       0 2862.58    26.1 2849.47    55.4 2825.29    78.6 2810.91   163.5 2765.15
   177.1 2756.06     189 2752.58   199.1 2744.13   213.4 2740.58   245.6 2723.19
   254.4 2716.55   271.1 2714.62   316.4 2692.04   368.9 2657.41   395.6    2631
   423.8 2630.69   435.3 2629.35     455 2633.39   480.2 2632.32   486.4    2634
   514.7 2657.57   531.7 2668.59     610 2709.24   621.9 2717.26   632.6 2720.56
   683.3 2753.71   746.3 2784.96     770 2791.25   785.9 2800.92   836.1 2822.59
#Mann= 5 ,-1 , 0
       0      .1       0  255.01     .06       0  374.68      .1       0
   395.6    .045       0   423.8      .1       0
#XS Ineff= 2 , 0
                          462.47         2639.28
Permanent Ineff=
       F       F
Bank Sta=395.6,423.8
XS Rating Curve= 0 ,0
Exp/Cntr=0.3,0.1

Type RM Length L Ch R = 1 ,23213   ,292.1,300,304
XS GIS Cut Line= 3
2409930.88656023656968.828094022     2410122.531      656613.787
      2410352.59      656238.408
#Sta/Elev= 30
       0 2849.56    47.7 2822.09    61.3 2805.01   109.2  2780.2   129.5 2767.16
     143 2763.65   193.1 2730.12   234.5  2705.5   243.4 2698.17   258.2 2694.99
   279.5 2682.08   319.7 2648.29   338.6 2629.27   347.7 2625.28     384 2617.69
   403.5 2615.82   414.5 2618.17   434.5 2616.81   440.6 2618.13   472.5 2637.33
   491.3  2646.6   538.2 2664.78   585.1 2687.43   603.9 2693.38   641.3 2714.35
     653 2719.21     754  2782.8   766.4 2786.36   792.6 2800.93   843.7 2823.77
#Mann= 5 ,-1 , 0
       0      .1       0  217.15     .06       0  380.04      .1       0
     384    .045       0   414.5      .1       0
Bank Sta=384,414.5
XS Rating Curve= 0 ,0
Exp/Cntr=0.3,0.1

Type RM Length L Ch R = 1 ,22913   ,303.6,300,295
XS GIS Cut Line= 3
2410014.56276885657016.681838389     2410357.576      656768.391
     2410705.237      656553.889
#Sta/Elev= 30
       0 2827.12      94 2764.79   110.3  2759.9   170.4 2723.72   202.7 2702.85
   212.6 2692.78   221.4 2687.65   230.6 2679.52   247.8 2675.46   271.8 2660.02
   287.9 2652.28   340.9 2616.67   355.8 2610.55   391.9 2607.11   407.62604.014
   434.1 2603.75   457.4 2601.72   463.2 2603.69   476.5 2619.88   485.9 2627.49
   525.3 2637.51   542.3 2644.94   553.3 2646.42     632 2682.56   657.9 2697.13
     688 2711.81   736.4 2742.49   749.1 2746.96   767.9  2760.1     832 2792.78
#Mann= 5 ,-1 , 0
       0      .1       0  175.47     .06       0  301.41      .1       0
   407.6    .045       0   434.1      .1       0
Bank Sta=407.6,434.1
XS Rating Curve= 0 ,0
Exp/Cntr=0.3,0.1

Type RM Length L Ch R = 1 ,22613   ,290.5,300,305.8
XS GIS Cut Line= 3
     2410371.585      657361.961     2410547.269      656997.042
 2410751.3349421656616.700985526
#Sta/Elev= 30
       0 2791.61    73.6 2760.13   145.5 2725.42   151.5 2718.24     164 2696.11
   173.3 2687.31   220.9  2666.4   238.4 2654.11     252 2652.44   283.9 2635.68
   339.3 2615.62   380.8 2594.11   397.52582.354   400.2 2582.16   412.52582.469
   429.8 2582.59   448.3 2588.71   471.2  2591.4   494.8 2603.34   530.3 2614.95
   589.4 2643.51   602.6 2651.64     616 2655.12     639 2666.25     648 2673.24
   720.7 2710.86   752.4 2732.36   769.6 2737.98   793.2 2753.71   836.6 2778.46
#Mann= 5 ,-1 , 0
       0      .1       0  173.62     .06       0  292.03      .1       0
   397.5    .045       0   412.5      .1       0
Bank Sta=397.5,412.5
XS Rating Curve= 0 ,0
Exp/Cntr=0.3,0.1

Type RM Length L Ch R = 1 ,22313   ,109.2,113.1,113.7
XS GIS Cut Line= 3
2410414.69492763657397.665932453     2410767.539      657159.156
     2411122.527      656956.954
#Sta/Elev= 30
       0  2770.9    26.4 2757.51   102.9 2711.32   106.3 2708.74   119.2 2692.72
   130.4 2683.63   176.4 2657.46   186.4  2650.1   200.8 2647.13   270.4 2614.39
   280.1 2612.25   323.5 2594.43   356.4 2583.37   381.5 2567.95   404.9 2563.15
   425.5    2562   440.2 2563.63     448 2568.27   475.4 2578.04   535.5 2617.15
   622.9 2659.54   636.6 2666.89   650.5    2677   663.1 2680.93   673.6 2689.09
   719.6 2709.25   779.4 2744.65   788.6 2760.92   793.3 2767.14   834.4 2784.44
#Mann= 5 ,-1 , 0
       0      .1       0  133.05     .06       0   242.5      .1       0
   404.9    .045       0   440.2      .1       0
Bank Sta=404.9,440.2
XS Rating Curve= 0 ,0
Exp/Cntr=0.3,0.1

Type RM Length L Ch R = 1 ,22200   ,331.7,336.9,339.4
XS GIS Cut Line= 3
 2410437.8410818657458.5625939432410652.91133869657335.766704695
2411198.03991061657081.657292265
#Sta/Elev= 30
       0 2778.52    71.9 2741.54    88.1 2723.59   111.6  2710.4   116.2 2705.71
   125.4 2690.65     130 2686.68   199.1 2647.02   211.5 2645.23   249.7 2627.09
   351.2 2586.38   388.2 2563.73   399.7 2559.96   416.12559.187   421.8 2558.69
   448.5  2559.6     458 2565.32     488 2567.79   505.4  2574.4   532.6 2595.34
   574.8 2623.74   593.9 2629.32   624.8 2647.93   642.5 2656.15   656.1 2657.98
     691 2677.36   770.4 2713.16   779.9 2721.08   800.5 2729.38   849.1 2758.46
#Mann= 5 ,-1 , 0
       0      .1       0   249.7     .06       0   351.2      .1       0
   416.1    .045       0   448.5      .1       0
Bank Sta=416.1,448.5
XS Rating Curve= 0 ,0
Exp/Cntr(USF)=0,0
Exp/Cntr=0.3,0.1

Type RM Length L Ch R = 1 ,21863   ,300,300,296.4
XS GIS Cut Line= 3
 2410506.8472335657634.527887171     2410956.776      657547.737
2411381.60891017657463.857432713
#Sta/Elev= 30
       0  2792.1    24.3 2772.73    65.1 2745.14   101.7 2716.73   130.3 2697.03
   179.1 2668.15   252.5 2631.55   268.8 2620.74   286.5 2618.07   305.4 2608.08
   362.5 2585.93     391 2570.57   419.6 2549.67   443.6 2540.54   452.1 2539.09
   476.5 2540.41   484.7 2539.98   500.3 2543.13   513.2 2549.32   533.6 2553.11
   574.4  2575.8   615.2 2590.03   627.3 2596.03   643.7 2597.93   709.2 2627.21
   736.4 2642.14   751.7 2647.02   814.9 2679.34   875.6 2707.86   891.3 2716.87
#Mann= 5 ,-1 , 0
       0      .1       0  266.43     .06       0  365.79      .1       0
   443.6    .045       0   476.5      .1       0
Bank Sta=443.6,476.5
XS Rating Curve= 0 ,0
Exp/Cntr=0.3,0.1

Type RM Length L Ch R = 1 ,21563   ,404.9,399.3,391.3
XS GIS Cut Line= 3
2410608.76760919657913.211787708     2411090.353      657790.925
      2411489.13      657699.375
#Sta/Elev= 30
       0 2762.29   158.2 2661.45   237.2 2615.81   278.5 2593.97   303.8 2583.46
   319.8 2575.15   336.3 2572.91   369.3 2563.61     390 2556.09   435.4 2532.73
   443.6 2530.98   472.5 2530.99   477.5 2529.56   484.9 2524.53     489 2522.51
   497.3 2521.69   513.3 2523.97   546.5 2527.24     567 2539.69   624.1  2563.1
   660.8 2580.62   669.6 2586.18   690.2 2588.75   718.9 2600.25   755.8 2619.63
   809.2  2643.3     821 2649.77   829.7 2651.91     842 2659.54     906 2691.37
#Mann= 5 ,-1 , 0
       0      .1       0  310.82     .06       0  410.52      .1       0
   484.9    .045       0   513.3      .1       0
Bank Sta=484.9,513.3
XS Rating Curve= 0 ,0
Exp/Cntr=0.3,0.1

Type RM Length L Ch R = 1 ,21164   ,337.7,350.7,357.2
XS GIS Cut Line= 3
2410959.32920747658405.1353039632411273.08720747658142.183303963
2411601.08420747657895.832303963
#Sta/Elev= 30
       0 2636.14     9.7 2631.24    28.4 2626.76    78.2 2605.41   145.4 2580.59
     163 2575.73   197.6 2570.85     209 2565.31   236.8 2547.49   256.7 2546.34
   270.6  2541.7     290 2539.31   313.5 2541.57   339.8 2548.58   348.9 2548.18
   359.3 2541.85   395.8 2511.15   401.9 2508.14   411.4 2506.67   441.4 2507.24
   471.5 2508.11   491.5 2506.63   501.5 2507.97     510 2511.79   556.5 2544.47
   572.9 2547.24   591.5 2556.65   607.2 2558.39   634.7 2568.47   819.6    2657
#Mann= 5 ,-1 , 0
       0      .1       0  181.11     .06       0  395.95      .1       0
   401.9    .045       0   441.4      .1       0
Bank Sta=401.9,441.4
XS Rating Curve= 0 ,0
Exp/Cntr=0.3,0.1

Type RM Length L Ch R = 1 ,20813   ,154.3,150,142.2
XS GIS Cut Line= 4
     2411011.769       658480.912411183.42894969658377.852560834
     2411461.894      658406.6062411748.71614576658448.416174409
#Sta/Elev= 30
       0 2643.71    45.5 2621.24    68.8 2606.36    87.5 2601.23   104.9 2590.15
   143.4 2570.29   171.4 2559.12   187.3 2555.08   235.7 2548.06     292 2537.39
   328.2 2532.69   340.3 2527.74   376.5 2504.44   396.6 2500.35   412.7 2491.57
   428.7 2488.67   448.9 2489.26   463.72487.282     477 2484.27   489.1 2484.95
     495 2487.94   501.2 2493.08   553.8 2492.21     578 2497.83   606.3 2498.13
   638.7 2494.39   654.8 2494.72   679.1 2504.05   723.6 2528.44     770 2546.64
#Mann= 5 ,-1 , 0
       0      .1       0  216.14     .06       0  421.88      .1       0
   463.7    .045       0     495      .1       0
Bank Sta=463.7,495
XS Rating Curve= 0 ,0
Exp/Cntr=0.3,0.1

Type RM Length L Ch R = 1 ,20663   ,298.2,300,306.6
XS GIS Cut Line= 3
     2411042.495      658670.098     2411418.577      658545.287
2411662.60250508658461.578264239
#Sta/Elev= 30
       0 2688.33    17.1 2678.98    59.3 2651.98    88.8 2635.02   198.3 2574.59
   240.1 2554.68   251.5 2547.58   265.8 2544.21   278.4 2537.42     316 2522.93
   344.5 2516.53   354.3 2508.59   366.9 2493.87   376.1 2485.54   382.5 2481.16
   388.8 2479.98   410.9 2481.01   421.8 2483.38   434.5 2483.33   455.6 2485.98
   464.1 2489.74   468.3 2490.51   493.7 2488.39   519.1 2490.12   557.1 2488.86
     591 2493.35   620.6 2491.78     629  2492.3   645.9 2494.77   654.2 2497.94
#Mann= 4 ,-1 , 0
       0      .1       0  304.45     .06       0   382.5    .045       0
   410.9      .1       0
Bank Sta=382.5,410.9
XS Rating Curve= 0 ,0
Exp/Cntr=0.3,0.1

Type RM Length L Ch R = 1 ,20363   ,263.5,262.2,256.2
XS GIS Cut Line= 3
2411151.30798361658848.320698868     2411589.015      658742.436
     2411995.897      658651.408
#Sta/Elev= 30
       0 2669.42    15.9 2659.34    32.3 2651.27    40.6 2645.05   106.4 2604.91
   184.6 2559.91   242.2 2528.79     304  2498.5   332.8 2491.91   361.6 2488.75
   378.5 2482.77   391.7 2474.72     411 2470.78   435.7 2468.77   450.3 2467.15
   476.7 2467.77   480.8 2469.17     489 2474.58   497.2 2476.87   558.8 2473.57
   587.4 2475.41   599.7 2477.61   612.2 2483.58   624.3 2491.31   665.2 2524.58
     698 2546.39   709.3 2553.14   726.7  2560.9   747.2 2574.67   867.3 2615.56
#Mann= 5 ,-1 , 0
       0      .1       0  321.95     .06       0  421.56      .1       0
   435.7    .045       0   480.8      .1       0
Bank Sta=435.7,480.8
XS Rating Curve= 0 ,0
Exp/Cntr=0.3,0.1

Type RM Length L Ch R = 1 ,20101   ,336.5,337.8,337.2
XS GIS Cut Line= 3
2411302.84978217659117.2492944122411703.31378217658966.175294412
2412087.43240759658829.453081981
#Sta/Elev= 30
       0 2611.87    94.9  2566.4   102.5 2562.07   179.4 2527.06   230.7 2499.11
     256 2487.38   286.3 2466.72   294.9 2462.17   301.3 2460.64   307.7 2460.15
   316.3 2460.49   333.4 2463.01   349.4 2460.77   367.6 2460.57   383.6 2457.05
   408.4 2459.22   421.4 2457.67   449.7 2456.53   452.9 2456.24   474.1 2463.84
   489.6 2473.26   525.1 2492.61   606.2 2526.22   673.7 2553.34   690.7 2558.75
   720.4 2571.27   746.4 2583.36   788.3 2606.03     801  2609.5   835.7 2621.34
#Mann= 5 ,-1 , 0
       0      .1       0  218.82     .06       0  340.15      .1       0
   421.4    .045       0   449.7      .1       0
#XS Ineff= 2 , 0
          332.05 2467.34
Permanent Ineff=
       F       F
Bank Sta=421.4,449.7
XS Rating Curve= 0 ,0
Exp/Cntr=0.3,0.1

Type RM Length L Ch R = 1 ,19763   ,294.6,300,302.7
XS GIS Cut Line= 3
     2411417.281      659402.621     2411816.176      659276.983
2412221.86962586659152.038006279
#Sta/Elev= 30
       0 2573.07    47.7 2550.77    81.2 2537.22    90.3  2534.6   169.3 2504.37
     221 2481.54   253.2 2468.78     288 2451.37   303.9 2447.22     337 2444.39
   362.2 2444.32   377.3 2440.95   399.6 2440.67   404.1 2439.01   408.3 2437.73
   416.7 2437.36   429.3 2437.76   434.7 2439.12   441.8 2442.24   458.6 2452.72
   471.1 2457.63   492.3 2469.37     513 2479.26   588.3 2511.22   651.1 2536.64
   681.1 2554.92     693 2561.06   722.3 2570.86   797.6 2606.09   842.7 2623.63
#Mann= 5 ,-1 , 0
       0      .1       0  249.08     .06       0  349.45      .1       0
   404.1    .045       0   434.7      .1       0
Bank Sta=404.1,434.7
XS Rating Curve= 0 ,0
Exp/Cntr=0.3,0.1

Type RM Length L Ch R = 1 ,19463   ,285.6,281.1,273.2
XS GIS Cut Line= 3
     2411438.947       659557.64     2411880.347      659563.229
2412283.40532517  659549.9110339
#Sta/Elev= 30
       0 2568.55    51.8 2539.69    83.8 2529.09   183.8 2488.19   223.8 2473.68
   267.8  2460.2   311.8 2444.67   347.8  2438.3   375.8 2427.84   387.8 2426.01
   407.7 2428.99   419.8 2428.94     428 2424.94   435.8 2421.85   443.8 2421.53
   453.82424.695   467.8    2435   475.9 2439.28   499.9 2442.45   507.9 2444.85
   571.9  2471.7   619.9 2487.95   635.9 2495.09   654.7 2500.22   675.3 2509.18
   688.2  2512.8     724 2526.45     760 2542.47     800 2552.89   844.7 2569.79
#Mann= 5 ,-1 , 0
       0      .1       0  354.55     .06       0     428    .045       0
   453.8     .06       0  455.28      .1       0
#XS Ineff= 2 , 0
          412.73 2437.31
Permanent Ineff=
       F       F
Bank Sta=428,453.8
XS Rating Curve= 0 ,0
Exp/Cntr=0.3,0.1

Type RM Length L Ch R = 1 ,19182   ,316.7,318.9,321.5
XS GIS Cut Line= 2
2411443.50594162659944.1580734442412275.54667483659686.241131826
#Sta/Elev= 30
       0  2572.2      62 2539.96    99.7 2525.69   124.8 2517.69   166.7 2499.93
   208.6 2485.61   301.5 2457.87   332.9 2446.87   355.3 2434.86   359.4 2431.75
   371.9 2418.51   374.4  2416.9   384.5 2415.49     3942410.136   409.6 2408.22
   428.8 2409.64   447.3 2413.49   468.2 2416.03   479.9  2418.9   497.5 2420.18
   514.3 2422.93   537.5  2428.8   560.4 2437.77   598.7 2455.52     619 2462.77
   673.4  2479.5   740.4 2504.26   786.5 2523.46   831.6 2545.84   871.1 2559.39
#Mann= 4 ,-1 , 0
       0      .1       0  310.31     .06       0     394    .045       0
   428.8      .1       0
Bank Sta=394,428.8
XS Rating Curve= 0 ,0
Exp/Cntr=0.3,0.1

Type RM Length L Ch R = 1 ,18863   ,300.4,300,298.1
XS GIS Cut Line= 3
2411529.07533921 660068.80398301     2411967.229      660094.232
2412377.48453373660138.770780847
#Sta/Elev= 30
       0 2539.66    41.4 2522.08   149.9 2480.44     194 2461.92     206 2458.13
   270.1 2429.01   286.2 2425.24   294.2 2421.51   321.7 2416.26   355.7 2398.88
   362.3  2397.7   378.3  2398.9   398.3  2396.4   431.5 2397.38   442.4 2395.38
   451.1 2396.97   462.5 2402.71   486.7 2409.39   498.8 2414.35   518.9 2425.28
     543 2441.04   569.7 2453.87   627.2 2476.29   667.7 2494.53     731 2519.21
   772.4  2537.5   792.5 2544.93   816.5 2552.14   824.7 2553.41   851.6 2566.48
#Mann= 5 ,-1 , 0
       0      .1       0  350.42     .06       0   431.5    .045       0
   451.1     .06       0  452.33      .1       0
#XS Ineff= 2 , 0
          374.56 2401.39
Permanent Ineff=
       F       F
Bank Sta=431.5,451.1
XS Rating Curve= 0 ,0
Exp/Cntr=0.3,0.1

Type RM Length L Ch R = 1 ,18563   ,299.6,300,301.4
XS GIS Cut Line= 3
2411575.09928697660406.582826307     2411986.619      660387.965
     2412395.217      660373.806
#Sta/Elev= 30
       0 2506.34    55.7 2482.66    71.2 2478.03   123.8 2457.96   203.9 2415.53
   219.9 2411.96   235.9 2403.83   247.9 2401.11   263.9 2401.51   295.9 2398.33
     332 2383.74   363.3 2382.53     388 2384.16   405.4 2382.52   420.1 2379.94
   432.4 2381.89     444 2389.04   452.1 2391.56   472.1 2400.64   500.1 2415.26
   516.1 2424.37   544.1  2443.3   628.2 2474.47   672.2  2492.7   712.2 2512.25
   724.3 2515.06   734.2 2521.27   768.3 2538.42   800.3 2551.65   820.8 2561.38
#Mann= 5 ,-1 , 0
       0      .1       0  253.08     .06       0   405.4    .045       0
   432.4     .06       0   453.1      .1       0
Bank Sta=405.4,432.4
XS Rating Curve= 0 ,0
Exp/Cntr=0.3,0.1

Type RM Length L Ch R = 1 ,18263   ,299.3,300,301.7
XS GIS Cut Line= 3
     2411593.113      660684.963     2412002.607      660687.178
     2412412.101      660689.393
#Sta/Elev= 30
       0 2487.45    45.6 2463.62    73.6 2451.08   162.7 2418.37   197.6 2403.66
   209.6 2400.33   249.6  2382.7   269.6 2381.08   337.5 2383.34   349.6 2379.71
   361.7 2378.19     4022369.378   409.6 2367.75     430 2367.95   437.6 2369.55
   457.6 2378.74   470.3    2381   485.6 2389.31   506.5 2403.14   549.6 2434.56
   561.6 2441.63   585.6 2452.48   601.6 2456.01   633.6 2470.59   673.6 2490.75
   725.6 2509.78   773.6 2531.58   789.6 2536.16   801.6  2543.4     819  2551.2
#Mann= 5 ,-1 , 0
       0      .1       0  181.34     .06       0  382.75      .1       0
     402    .045       0   437.6      .1       0
Bank Sta=402,437.6
XS Rating Curve= 0 ,0
Exp/Cntr=0.3,0.1

Type RM Length L Ch R = 1 ,17963   ,304.1,300,293.7
XS GIS Cut Line= 3
2411571.33786092660956.762695405     2411991.377      660986.241
     2412398.019      661020.221
#Sta/Elev= 30
       0 2493.41    38.9 2476.31   151.8 2417.68   173.9 2402.64   199.9 2382.61
   215.9  2372.1     224 2368.49     240 2366.82   268.1 2370.06   284.1 2366.58
   297.4 2360.14   308.2 2357.88   340.2 2361.31   400.4 2360.47   408.4 2357.59
   424.5 2355.58   439.6 2357.97   444.5 2361.53   456.6 2375.84   460.6 2378.19
   480.4 2382.29   508.7 2394.62   520.8 2397.46   564.9 2423.53     593 2438.18
   693.4 2478.06   757.6 2506.82   765.6 2511.71   797.7 2520.89   829.1 2537.01
#Mann= 5 ,-1 , 0
       0      .1       0  148.46     .06       0  352.51      .1       0
   408.4    .045       0   439.6      .1       0
#XS Ineff= 2 , 0
           350.1 2373.79
Permanent Ineff=
       F       F
Bank Sta=408.4,439.6
XS Rating Curve= 0 ,0
Exp/Cntr=0.3,0.1

Type RM Length L Ch R = 1 ,17663   ,294.8,300,304.5
XS GIS Cut Line= 3
     2411554.614      661429.271     2411926.216      661269.152
2412335.76920013661133.111887352
#Sta/Elev= 30
       0 2454.67   122.1 2408.57   139.5    2406   157.2 2401.21   183.1 2390.61
   199.8 2386.07   244.1  2370.8   274.5 2356.56   322.5 2350.77     366 2347.92
   385.4 2348.64   387.8  2348.4   393.7 2344.74   397.6 2342.43   405.2 2341.55
   419.5 2344.94   426.3 2346.17   443.1 2345.82   451.6 2347.57   468.4 2347.41
   493.7 2360.13   506.3  2363.3   531.6  2366.6   556.9 2374.03   615.7 2398.03
   640.2  2409.4   683.4 2426.53     734 2449.54   780.3 2476.57   836.2 2505.78
#Mann= 5 ,-1 , 0
       0      .1       0  244.01     .06       0   393.7    .045       0
   419.5     .06       0  448.04      .1       0
Bank Sta=393.7,419.5
XS Rating Curve= 0 ,0
Exp/Cntr=0.3,0.1

Type RM Length L Ch R = 1 ,17363   ,301.9,300,295.1
XS GIS Cut Line= 3
     2411563.233      661536.679     2411972.416      661552.599
     2412381.824      661563.101
#Sta/Elev= 30
       0 2440.45    15.5 2438.61    43.5 2431.26    59.6 2430.06    79.6 2422.88
   115.6 2412.75   135.6 2411.22   179.6 2402.82   187.7 2399.06   203.7 2388.38
   223.7 2369.97   247.7 2352.23   267.7 2343.98   291.7 2340.78   359.6 2339.95
   371.8 2338.49   383.8 2334.53   395.8 2333.95   399.8 2332.18   403.8 2330.47
   411.8 2329.74   419.8 2329.89   426.62332.247   447.8 2345.81   463.8 2354.29
   479.8 2355.75   495.9 2362.56   561.5 2381.28   731.9 2438.35     819 2463.53
#Mann= 5 ,-1 , 0
       0      .1       0  351.64     .06       0   399.8    .045       0
   426.6     .06       0  452.86      .1       0
Bank Sta=399.8,426.6
XS Rating Curve= 0 ,0
Exp/Cntr=0.3,0.1

Type RM Length L Ch R = 1 ,17063   ,297.5,300,302.6
XS GIS Cut Line= 3
     2411614.184      661926.107       2412035.6      661837.107
2412448.03388672661734.353112648
#Sta/Elev= 30
       0  2458.9    70.1  2438.8     111 2425.09   209.1 2388.22   221.3 2382.04
   233.6 2378.08   249.6 2368.35   278.6 2343.52   290.8 2334.11   310.3 2323.78
   315.4 2322.73   331.7 2322.69   352.2 2327.03   364.4 2326.38   381.2 2322.31
     389    2322   402.7 2323.63   413.5 2321.11   438.1 2319.08   442.2 2319.34
   448.3 2321.64   458.7 2328.99   483.4 2354.14   495.8  2362.5     504 2365.98
   527.5 2368.93   578.2 2372.54   682.6  2387.7     772 2407.45   855.8 2431.26
#Mann= 5 ,-1 , 0
       0      .1       0  357.09     .06       0   413.5    .045       0
   448.3     .06       0  456.58      .1       0
#XS Ineff= 2 , 0
          353.12 2330.51
Permanent Ineff=
       F       F
Bank Sta=413.5,448.3
XS Rating Curve= 0 ,0
Exp/Cntr=0.3,0.1
