HEC-RAS study BRUSHRN.prj: BRUSHRN

--- BRUSHRN.g01 (geometry) --- (continued)

Type RM Length L Ch R = 1 ,16763   ,91,88.5,84.5
XS GIS Cut Line= 3
2411602.96547829 662171.99014726     2412003.674      662119.436
     2412459.849      662060.257
#Sta/Elev= 30
       0 2467.29    57.8 2431.16    72.1 2423.31   111.3 2406.53   161.3 2387.48
   230.6 2353.38   290.2 2331.15   338.7 2322.26   354.8 2316.32   370.9 2315.09
   389.5 2304.65   395.1 2302.57   407.1 2302.14   415.3 2304.94   423.4 2308.78
   427.4 2309.35   459.7 2310.64   479.8 2314.24   508.1 2313.94   520.2 2318.14
   544.4 2323.26     568 2338.71   576.6 2342.66   588.7 2346.08   689.6 2355.12
     738 2361.69   746.1 2365.74   758.2 2368.06   782.4 2376.98   864.1 2420.82
#Mann= 4 ,-1 , 0
       0      .1       0  307.94     .06       0   389.5    .045       0
   415.3      .1       0
Bank Sta=389.5,415.3
XS Rating Curve= 0 ,0
Exp/Cntr=0.3,0.1

Type RM Length L Ch R = 1 ,16674   ,22.4,22.6,22.8
XS GIS Cut Line= 3
2411679.31384945662354.2837836122412244.73137896662098.463080723
2412422.96081761662078.489091908
#Sta/Elev= 30
       0 2409.59    83.7 2377.06   171.4 2355.23   240.9 2329.71   262.8  2324.5
   297.9 2319.51   319.9 2308.68   337.7 2308.49   341.8 2306.91   347.9 2301.78
   350.6  2299.7   357.6 2298.34   370.9 2301.22   381.3 2307.58   385.7 2308.32
   416.5 2306.79   438.4 2309.92   483.7 2308.14   504.3 2309.41     513 2311.91
   528.1 2319.38   543.2 2330.25     557 2333.59   565.7 2341.28   570.1 2343.13
   592.1 2346.65   658.8 2353.05   711.2  2360.8   751.4 2375.41   799.9 2400.31
#Mann= 5 ,-1 , 0
       0      .1       0  271.01     .06       0   347.9    .045       0
   370.9     .06       0  402.07      .1       0
Bank Sta=347.9,370.9
XS Rating Curve= 0 ,0
Exp/Cntr(USF)=0,0
Exp/Cntr=0.5,0.3

Type RM Length L Ch R = 1 ,16652   ,49.2,49.2,48.8
XS GIS Cut Line= 3
2411680.85031013 662378.86715446 2412255.4866037662117.668839198
2412408.36444116662102.304232418
#Sta/Elev= 30
       0 2406.25    86.9 2374.79   111.9    2368     191 2351.74   212.9  2345.8
   270.1 2326.72   300.9 2319.36   309.3 2314.78   318.9 2307.03     336 2305.65
   349.2 2306.35     358 2300.61   362.4 2298.38   369.9 2297.87     379 2298.56
   384.3  2300.6   393.1  2305.2   419.5 2305.61   445.5 2308.31     521 2307.84
   542.5 2317.47   563.3 2333.41   569.3 2336.53   581.4 2338.23   593.5  2342.9
   617.6 2347.02   646.5 2348.94   703.3 2356.91     739 2370.74   784.9 2393.36
#Mann= 5 ,-1 , 0
       0      .1       0  273.65     .06       0     358    .045       0
   384.3     .06       0  479.51      .1       0
#XS Ineff= 2 , 0
           350.2    2302   393.1            2302
Permanent Ineff=
       F       F
Bank Sta=358,384.3
XS Rating Curve= 0 ,0
Exp/Cntr(USF)=0,0
Exp/Cntr=0.5,0.3

Type RM Length L Ch R = 1 ,16603   ,141.6,139.8,140.4
XS GIS Cut Line= 2
 2411700.4746669662432.1262068332412344.08097314662122.273303433
#Sta/Elev= 30
       0 2394.86    20.6 2387.32    42.5 2380.94   104.6 2366.58   170.4 2357.05
   233.4 2351.31     260 2345.81   270.3 2342.25   277.8 2338.09   308.8 2314.08
   322.2 2305.58     331 2303.44   359.2 2302.64   371.2  2299.4   380.2 2296.36
   388.7 2295.86   393.2  2296.4   398.2 2298.78   406.5 2301.39   428.2 2302.15
   468.7 2306.71   517.5 2306.12   530.8 2307.28   548.6 2313.98   588.5 2336.65
   597.4 2340.67   619.6 2342.39   639.1  2346.4   668.4 2350.47   714.3 2362.49
#Mann= 5 ,-1 , 0
       0      .1       0  310.58     .06       0   371.2    .045       0
   398.2     .06       0  471.22      .1       0
Bank Sta=371.2,398.2
XS Rating Curve= 0 ,0
Exp/Cntr(USF)=0,0
Exp/Cntr=0.5,0.3

Type RM Length L Ch R = 1 ,16463   ,298.2,300,301.7
XS GIS Cut Line= 3
2411795.11586973662599.093200126     2412151.642      662355.794
     2412493.954      662133.259
#Sta/Elev= 30
       0 2360.98    28.6 2357.74   128.1 2352.42   193.3 2345.32   238.8 2338.75
   280.4 2331.44   319.2 2322.47   359.7 2309.75   385.6 2297.02   405.7 2295.79
   411.9 2296.65   418.82294.119   425.7 2292.65   444.9 2292.33   449.6 2292.81
   452.8 2294.24   460.5 2297.08   480.8 2294.96   506.9    2299   521.4 2307.62
   532.8 2315.69   554.6 2327.32   568.9 2332.74   613.8 2347.17   653.5 2358.41
     660 2361.98   748.9  2397.2     767 2405.89   804.6 2421.74   839.9 2438.39
#Mann= 4 ,-1 , 0
       0      .1       0   315.6     .06       0   418.8    .045       0
   452.8      .1       0
Bank Sta=418.8,452.8
XS Rating Curve= 0 ,0
Exp/Cntr=0.3,0.1

Type RM Length L Ch R = 1 ,16163   ,293.4,300,308.5
XS GIS Cut Line= 3
     2411929.533      662803.292     2412298.776      662616.089
 2412653.8393304662426.152895531
#Sta/Elev= 30
       0 2336.34    32.8 2333.73    82.1 2327.24    95.5 2324.57   132.1 2314.14
   155.9 2308.69   171.8  2308.3   197.6 2305.51   225.6  2306.7   261.5 2304.74
     275 2301.58   301.8 2290.12   328.2  2282.7   379.1 2283.63   388.1 2282.99
     400 2280.21   409.5 2277.59   418.5 2277.66   430.5 2280.35   441.2 2283.59
   459.3  2295.4   491.1 2313.74   527.4 2341.49   559.1 2361.37   604.5 2384.04
   627.6 2397.98   730.3 2447.28   763.3 2462.02   801.2 2480.87   816.7 2489.76
#Mann= 5 ,-1 , 0
       0      .1       0     329     .06       0     400    .045       0
   430.5     .06       0   508.4      .1       0
Bank Sta=400,430.5
XS Rating Curve= 0 ,0
Exp/Cntr=0.3,0.1

Type RM Length L Ch R = 1 ,15863   ,328.4,325.9,317.7
XS GIS Cut Line= 3
     2411951.617      662889.195     2412358.242      662903.277
2412784.93507119662920.663622037
#Sta/Elev= 30
       0 2325.82    87.2 2314.07   163.2 2298.03   204.6 2292.62   219.3 2292.41
   235.3 2290.14   271.3 2291.98   315.3 2290.64   335.3 2282.81   347.3 2270.23
   351.3 2268.06   364.4  2267.7   379.4 2270.15   395.4 2263.95   395.4 2263.94
   403.1 2261.63   411.4 2261.42   423.4 2264.04   431.4 2270.73   435.4 2272.55
   463.4 2272.82   495.5 2270.38   519.5 2276.29   567.5 2308.41   583.5 2317.69
   607.5 2324.38   643.6 2339.78   679.6  2358.4   735.6 2384.77   833.9 2427.85
#Mann= 7 ,-1 , 0
       0      .1       0   25.85     .05       0  282.44      .1       0
  383.68     .06       0   395.4    .045       0   423.4     .06       0
  485.02      .1       0
Bank Sta=395.4,423.4
XS Rating Curve= 0 ,0
Exp/Cntr=0.3,0.1

Type RM Length L Ch R = 1 ,15537   ,281.9,274.1,269
XS GIS Cut Line= 3
2412086.92153672663298.8347514112412513.96530339663160.915088701
2412899.91430339663039.738088701
#Sta/Elev= 30
       0 2303.14    16.6 2300.63    51.9 2299.04    88.1 2292.53   120.6 2285.29
   159.5 2285.02     182 2281.81   226.8 2279.04   260.4 2274.19   302.5 2271.99
   319.3 2267.38   336.1    2261   348.7 2261.08   365.2 2259.29   390.7 2252.26
   403.3 2251.57   412.9 2249.65     437 2249.96   449.6 2247.16     458  2247.5
   463.8 2249.61   478.9 2258.44   492.5 2261.32     525 2277.48   562.7 2293.78
     652  2339.7     764 2401.41   789.4 2411.78   822.7 2428.28   853.3 2441.67
#Mann= 5 ,-1 , 0
       0      .1       0  311.96     .06       0     437    .045       0
   463.8     .06       0  512.82      .1       0
Bank Sta=437,463.8
XS Rating Curve= 0 ,0
Exp/Cntr=0.3,0.1

Type RM Length L Ch R = 1 ,15263   ,603.3,600,588.6
XS GIS Cut Line= 3
     2412282.453       663674.43     2412599.562      663416.806
2412940.70876526663178.725147892
#Sta/Elev= 30
       0 2342.51      12 2339.63    51.9 2323.31   103.4 2305.89   136.4  2297.6
     162 2287.29   195.9 2270.37   213.1 2264.36     253 2260.52   278.5 2247.86
   287.1 2245.31   309.6 2242.81   334.9 2243.32   386.6 2237.72   411.9 2235.66
   423.7 2237.83   432.3  2245.9   438.1 2248.05   466.1 2248.95   486.9 2247.18
   519.8  2249.9   539.3 2249.75     549 2252.08   573.4 2266.87   635.6  2298.6
   705.3 2338.13   729.5 2352.14   763.6 2374.81   791.4  2390.7   824.6 2405.66
#Mann= 5 ,-1 , 0
       0      .1       0  316.93     .06       0   386.6    .045       0
   423.7     .06       0  430.61      .1       0
Bank Sta=386.6,423.7
XS Rating Curve= 0 ,0
Exp/Cntr=0.3,0.1

Type RM Length L Ch R = 1 ,14663   ,334,337.8,341.4
XS GIS Cut Line= 3
     2412840.752      664202.959     2412985.309      663814.641
     2413160.564      663436.043
#Sta/Elev= 30
       0 2273.34      14 2274.18    42.8 2277.12    68.4  2285.6   132.4 2288.15
     154 2280.09   170.8 2266.48   183.6 2262.75   192.1 2255.15   222.4 2235.69
     238 2229.05   264.7 2224.66   290.3 2217.95   311.6 2218.11   328.7 2221.19
   358.6 2215.91   393.5 2215.26   404.7 2211.13   418.3 2207.64   433.3 2211.13
   449.3 2219.18   458.2 2227.22   480.2  2252.3     489 2257.39   590.4 2264.02
   647.7 2272.39   674.9 2274.34   740.3 2291.01   806.9 2310.86   831.5 2315.12
#Mann= 6 ,-1 , 0
       0     .05       0      14      .1       0   73.76     .05       0
  297.34     .06       0   404.7    .045       0   433.3      .1       0
Bank Sta=404.7,433.3
XS Rating Curve= 0 ,0
Exp/Cntr=0.3,0.1

Type RM Length L Ch R = 1 ,14325   ,261.4,262.2,265.2
XS GIS Cut Line= 2
2412975.45113373664335.6161193092413514.21921345663680.677251135
#Sta/Elev= 30
       0 2291.41   104.5 2280.15   140.8 2272.18   200.4 2267.76   223.7 2263.19
   250.1 2255.59   265.1 2249.19   295.6 2225.15   306.5 2213.49   316.9 2208.64
   342.8 2201.19   358.3 2203.07   375.1 2202.46   384.2 2200.13   408.2 2200.98
   417.8 2195.45   429.1 2192.47   445.9 2195.14   463.2 2194.93   468.9 2196.28
   477.5 2200.98   505.9 2222.22   513.7 2225.72   666.3 2258.26   704.8  2284.7
   748.2 2306.89     767 2318.77   778.7 2323.84   829.8 2371.29   848.1  2383.1
#Mann= 5 ,-1 , 0
       0      .1       0  324.72     .06       0   417.8    .045       0
   445.9     .06       0  471.27      .1       0
Bank Sta=417.8,445.9
XS Rating Curve= 0 ,0
Exp/Cntr=0.3,0.1

Type RM Length L Ch R = 1 ,14063   ,339.8,345.2,357
XS GIS Cut Line= 3
     2413205.088      664440.566     2413483.713      664109.046
     2413732.129      663788.745
#Sta/Elev= 30
       0 2270.75       8 2268.12    30.8 2266.51    50.6 2260.83    75.3 2258.35
    87.5 2252.41   101.5 2251.24   113.1  2246.4   148.5 2237.69   164.2 2232.12
   226.4 2221.83   282.3 2200.45   294.8 2198.75   360.1 2198.19   378.4 2190.44
   406.7 2189.54   420.2 2184.33   436.8 2182.64   462.4 2184.02     471 2188.16
   493.8 2213.42   516.3 2229.83   557.3 2248.37   577.5 2259.57   607.8 2279.81
   653.4 2305.53   690.5 2322.76   730.4  2351.5   790.1 2391.65   838.4 2417.75
#Mann= 5 ,-1 , 0
       0      .1       0  371.17     .06       0   420.2    .045       0
   462.4     .06       0  504.74      .1       0
Bank Sta=420.2,462.4
XS Rating Curve= 0 ,0
Exp/Cntr=0.3,0.1

Type RM Length L Ch R = 1 ,13718   ,33.1,32.6,31.8
XS GIS Cut Line= 2
2413291.24272928664583.7786080482413996.40185961664231.925402012
#Sta/Elev= 30
       0 2267.69    17.3  2261.4    27.1 2259.05    48.6 2256.78    73.7 2247.51
    86.8 2245.26   124.6 2228.43   142.5 2227.31   154.3 2220.54   181.2 2209.37
     209 2194.03   218.5 2190.88   227.4 2186.13   267.7 2184.25   348.1 2172.83
   374.9    2173   379.4  2172.1   386.92167.271   392.8  2164.5   396.9 2164.27
   406.2 2164.74   416.6 2167.16   428.6 2171.99   438.7 2173.48   468.8 2190.77
   496.6 2199.85     546 2221.43   643.2 2255.87   656.4 2262.34   788.1 2315.91
#Mann= 6 ,-1 , 0
       0      .1       0  250.61     .05       0  352.28     .06       0
   386.9    .045       0   416.6     .06       0  453.86      .1       0
Bank Sta=386.9,416.6
XS Rating Curve= 0 ,0
Exp/Cntr=0.5,0.3

Type RM Length L Ch R = 1 ,13685   ,16.6,16.7,16.7
XS GIS Cut Line= 2
2413332.79984647664614.1479473272414014.19452863664242.132324786
#Sta/Elev= 30
       0 2262.43      25 2262.31    33.3 2257.56    56.9 2250.35    79.7 2241.25
   101.1 2238.95     107 2236.15   116.1 2229.52   130.6  2228.2   145.3 2219.04
     180 2203.14   198.2 2191.83   207.3 2184.99   234.6 2178.55   260.3 2177.74
   316.3 2171.29   348.6 2170.69   357.32165.569   362.2 2163.85   372.3 2163.67
   380.5 2164.22     3882166.874   398.7 2171.04   412.4 2172.46   458.4 2190.78
   526.3 2218.09   582.8 2236.66     704 2288.12   745.1  2304.7   776.3 2319.56
#Mann= 5 ,-1 , 0
       0      .1       0   260.3     .05       0   357.3    .045       0
     388     .06       0   458.4      .1       0
Bank Sta=357.3,388
XS Rating Curve= 0 ,0
Exp/Cntr(USF)=0,0
Exp/Cntr=0.5,0.3

Type RM Length L Ch R = 1 ,13668   ,32.8,32.7,32.8
XS GIS Cut Line= 2
2413334.01114323664630.8173681082414020.78299409664258.729448012
#Sta/Elev= 30
       0 2262.18    35.9    2260      60  2253.6    92.2 2241.91   114.6 2238.36
   128.2 2230.38   142.6 2228.78   169.2  2214.9     201 2195.72   215.9 2183.72
   232.9 2179.52   246.5 2179.13   269.2  2173.5   282.9 2172.54   314.7 2172.33
   351.1 2170.08   355.7 2168.86   361.52165.144   366.4 2163.55   377.7 2163.23
   392.22166.125   414.8  2170.2   423.9 2174.85   434.2 2177.57   453.3 2180.85
   481.4 2193.79   533.1 2213.89   602.4 2238.32   755.9 2305.45   781.1  2318.9
#Mann= 5 ,-1 , 0
       0      .1       0   282.9     .06       0   361.5    .045       0
   392.2     .06       0   434.2      .1       0
Bank Sta=361.5,392.2
XS Rating Curve= 0 ,0
Exp/Cntr(USF)=0,0
Exp/Cntr=0.5,0.3

Type RM Length L Ch R = 1 ,13636   ,179,172.8,166.2
XS GIS Cut Line= 2
2413359.43385487 664652.629608372414021.21143032664297.475642878
#Sta/Elev= 30
       0 2262.51    26.5 2259.45    80.9 2246.06   103.6 2242.89   124.9 2231.74
   139.9 2230.77   176.3 2207.79   189.9 2197.81   203.5 2185.12     208 2183.18
   225.3 2181.28   248.9 2172.87   291.3 2172.51   339.7 2168.16   346.8 2165.19
   353.3 2162.62   361.2 2162.26   371.5 2162.62   378.62164.697   384.8 2166.38
   393.7 2165.98   412.3 2172.04   423.2 2176.97   444.1 2179.35   460.5 2183.55
   539.4 2215.94   594.6 2234.82   618.2 2244.76   698.3 2284.14   751.1  2307.5
#Mann= 5 ,-1 , 0
       0      .1       0   291.3     .06       0   346.8    .045       0
   378.6     .06       0   412.3      .1       0
Bank Sta=346.8,378.6
XS Rating Curve= 0 ,0
Exp/Cntr(USF)=0,0
Exp/Cntr=0.3,0.1

Type RM Length L Ch R = 1 ,13463   ,300.5,300,300.6
XS GIS Cut Line= 3
     2413534.667      664918.644     2413795.343      664605.545
     2414071.072       664286.95
#Sta/Elev= 30
       0 2239.06    70.9 2226.84     109 2223.45   137.7  2224.1   190.2 2214.53
   233.9 2203.11   275.5 2183.87   293.9 2176.73   327.6 2172.28   352.1 2163.83
   374.4 2162.52   387.7 2156.83   395.2 2154.65   414.5 2153.96   420.2 2154.41
   424.8 2156.74   430.9 2159.92   437.1 2159.47   451.4  2161.1   469.1 2166.16
   504.3  2169.1   528.7 2181.59   564.3 2191.19   624.4 2218.62   666.9 2242.41
   693.8 2259.49   724.3 2276.96   748.8 2290.21   783.2 2306.86   828.8  2333.1
#Mann= 5 ,-1 , 0
       0      .1       0  306.16     .06       0   387.7    .045       0
   424.8     .06       0  443.79      .1       0
Bank Sta=387.7,424.8
XS Rating Curve= 0 ,0
Exp/Cntr=0.3,0.1

Type RM Length L Ch R = 1 ,13163   ,297.6,300,302.5
XS GIS Cut Line= 3
     2413677.121      665030.631     2414055.687      664742.833
2414353.65474242664511.738159659
#Sta/Elev= 30
       0 2268.62    62.3 2254.66   138.4 2240.86   212.2 2221.57     295 2172.65
   306.4 2163.72   320.7 2160.51   338.7 2150.75   444.2 2147.68   455.6  2145.6
   466.3 2138.88   474.8 2135.97   483.4 2136.88   488.5 2139.68     509  2145.5
     525 2147.25   534.7 2150.07   546.1 2156.65   568.9  2174.3   594.6 2181.86
   614.5 2193.17   641.4 2199.44   677.8 2217.44   723.5 2249.07   752.8 2271.03
   757.8 2273.86   768.5 2276.75   778.1 2285.45   816.9 2311.12   852.6  2330.4
#Mann= 5 ,-1 , 0
       0      .1       0  279.14     .06       0  460.28      .1       0
   466.3    .045       0   488.5      .1       0
Bank Sta=466.3,488.5
XS Rating Curve= 0 ,0
Exp/Cntr=0.3,0.1

Type RM Length L Ch R = 1 ,12863   ,329.7,325.7,321.5
XS GIS Cut Line= 3
     2413707.667      665128.517      2414102.03      665026.557
     2414509.794      664918.675
#Sta/Elev= 30
       0 2282.44    43.3 2271.32    94.1  2255.6   151.9  2227.9   200.8 2201.85
     280 2162.85   333.7  2144.7   351.8 2134.17   378.1 2132.45   387.9 2127.47
   391.5 2125.61   403.9 2124.71   420.5 2124.99   428.8 2127.33   441.2 2129.94
   457.7 2130.48   474.3  2136.1   486.7  2137.1   519.8 2150.27   528.1 2152.51
   569.4 2150.48   598.4 2151.09   623.6 2153.01   643.9 2156.82   693.6 2170.72
   767.6 2199.29   785.8 2208.23   805.3 2221.49   817.7 2225.32   829.1 2233.53
#Mann= 4 ,-1 , 0
       0      .1       0  293.73     .06       0   387.9    .045       0
   428.8      .1       0
Bank Sta=387.9,428.8
XS Rating Curve= 0 ,0
Exp/Cntr=0.3,0.1

Type RM Length L Ch R = 1 ,12537   ,282.5,274.3,266.7
XS GIS Cut Line= 3
2413878.06119131665498.2756085582414246.53019131665315.764608558
2414619.17119131665146.922608558
#Sta/Elev= 30
       0 2322.91    36.5 2302.06    76.6  2276.2   119.5 2254.09   144.4 2238.72
   182.1 2211.63   205.9 2198.91   232.9 2181.29   246.3 2171.57   262.7 2155.89
   295.6 2134.64     314 2126.02   328.4 2121.97   362.3 2121.96   389.1 2120.07
   411.4  2111.7   420.2 2109.32     429 2109.12   442.4 2111.05   451.3 2117.94
   468.5 2118.22   490.5 2122.71   499.3  2127.3   516.8 2140.51   622.2 2142.22
   653.8 2144.56     681 2148.78   736.4    2164   783.7 2182.69   820.3 2193.85
#Mann= 6 ,-1 , 0
       0      .1       0  399.85     .06       0   411.4    .045       0
   442.4     .06       0  502.86      .1       0  708.66      .1       0
Bank Sta=411.4,442.4
XS Rating Curve= 0 ,0
Exp/Cntr=0.3,0.1

Type RM Length L Ch R = 1 ,12263   ,328.6,336.3,342.4
XS GIS Cut Line= 3
     2414150.331      665869.548     2414393.187      665542.434
 2414654.2088842665221.999937277
#Sta/Elev= 30
       0 2268.92    45.1 2241.42    81.2 2214.21      88 2206.36    93.7 2201.11
   139.4 2171.97   162.7 2158.49   197.6 2144.71   259.5  2112.6   265.2 2111.14
   297.2  2108.1   376.5  2106.3   383.2 2104.64   389.9 2101.15   396.8 2098.93
     412 2098.74   417.1 2098.97   422.4 2101.17   441.5 2107.63   456.5 2107.45
   466.9 2109.27   476.9 2114.17   493.5 2124.39   527.6 2133.36   549.2 2136.67
     647 2145.02   686.8 2151.89   732.3 2163.21   762.8 2175.31   820.7 2189.02
#Mann= 6 ,-1 , 0
       0      .1       0  240.96     .06       0   379.5      .1       0
   389.9    .045       0   422.4      .1       0  797.18      .1       0
Bank Sta=389.9,422.4
XS Rating Curve= 0 ,0
Exp/Cntr=0.3,0.1

Type RM Length L Ch R = 1 ,11927   ,75.1,74.2,73.3
XS GIS Cut Line= 3
2414215.71624231665990.9233283132414585.13424231665789.416328313
2414960.04021819665612.189202868
#Sta/Elev= 30
       0 2238.47    26.2 2225.91    58.3 2213.25    67.2  2205.9    90.7 2191.64
   126.5 2165.57   167.4 2130.15   181.1 2113.97   190.3 2109.33   208.5 2103.79
   242.3 2103.65   275.7 2099.14   322.4 2098.66   334.2 2095.22   363.4  2091.5
   420.8 2092.48   426.9 2090.18   431.4 2086.28   438.9 2082.92   447.9 2082.32
     460 2085.78   484.5 2099.37     505 2103.06     520 2114.35   528.8 2118.58
   648.2 2117.81   710.2 2113.41   754.4 2125.05   785.4 2131.68   835.5 2145.79
#Mann= 5 ,-1 , 0
       0      .1       0  345.91     .06       0   431.4    .045       0
     460      .1       0  760.75      .1       0
Bank Sta=431.4,460
XS Rating Curve= 0 ,0
Exp/Cntr=0.5,0.3

Type RM Length L Ch R = 1 ,11852   ,27.4,27.3,27.2
XS GIS Cut Line= 2
2414280.66403734 666060.789266972414978.84713403665637.647996245
#Sta/Elev= 30
       0 2177.99    11.6 2172.11    23.3 2168.72    69.9 2149.11     104 2130.49
   111.7  2127.9   215.5 2107.65   264.4 2100.58   291.2  2098.7   302.9 2093.04
   320.1 2088.08   339.2 2089.88   376.6 2088.95     386 2087.92   395.3 2082.48
     400 2079.89   407.7 2079.02     414 2079.51   419.4 2082.64   437.4 2090.99
   474.7 2092.29   498.2 2110.95   505.3 2113.22   587.1 2112.97   681.5  2108.2
     706 2109.73   739.7 2118.62   764.8 2122.88   797.6  2135.4   816.4 2144.25
#Mann= 8 ,-1 , 0
       0      .1       0  294.82     .06       0   395.3    .045       0
   419.4     .06       0  447.76      .1       0  616.19     .05       0
  703.87      .1       0  723.32      .1       0
#XS Ineff= 2 , 0
             386    2088     431            2088
Permanent Ineff=
       F       F
Bank Sta=395.3,419.4
XS Rating Curve= 0 ,0
Exp/Cntr(USF)=0,0
Exp/Cntr=0.5,0.3

Type RM Length L Ch R = 1 ,11825   ,76.7,72.5,68.1
XS GIS Cut Line= 2
 2414295.1580663666086.733332873 2415002.0760663665652.620332873
#Sta/Elev= 30
       0 2164.13    41.8 2147.77    53.2  2138.9    69.9  2137.3   116.9 2126.43
   130.9 2124.91   182.8 2111.96   197.3 2109.27   215.4 2108.88   258.4 2101.97
   299.9 2098.23   318.7 2089.32   331.1 2087.64   386.4  2088.2   389.3 2087.62
   396.52081.741   400.6 2079.08   407.9 2078.27   417.3 2079.16   421.3 2081.37
   431.4 2087.87   435.8 2089.08   479.4  2090.5   488.9 2094.92   506.5 2107.91
   515.9 2110.73   581.2 2110.49   684.8 2105.94   764.1 2115.95   829.6 2148.39
#Mann= 7 ,-1 , 0
       0      .1       0  284.55     .06       0   396.5    .045       0
   421.3     .06       0  499.31      .1       0  606.69     .05       0
  766.16      .1       0
Bank Sta=396.5,421.3
XS Rating Curve= 0 ,0
Exp/Cntr=0.5,0.3

Type RM Length L Ch R = 1 ,11753   ,58,55.8,53.4
XS GIS Cut Line= 3
2414406.41910533666247.0175819512414799.32256243665802.073931862
2414951.54012693665699.294550702
#Sta/Elev= 30
       0 2247.76    36.8 2236.46    85.1 2217.38    96.2 2206.47   133.6 2186.82
     159 2168.66   176.3 2159.72   202.9 2135.87     218 2125.02   242.2 2110.28
     267 2097.94     283 2092.03   302.6 2087.53   338.9  2085.2   395.1 2086.15
   399.9 2084.59   405.4 2079.08   411.2 2075.99   416.9 2075.81   427.1 2076.73
   435.6 2079.86   443.1 2084.92   447.7 2086.44   507.6 2087.47   514.2  2089.7
   535.9 2103.22   544.4 2105.71     607 2107.86   698.5 2104.31   777.3 2114.04
#Mann= 6 ,-1 , 0
       0      .1       0   359.9     .06       0   405.4    .045       0
   435.6     .06       0  488.32      .1       0  613.32     .05       0
Bank Sta=405.4,435.6
XS Rating Curve= 0 ,0
Exp/Cntr(USF)=0,0
Exp/Cntr=0.5,0.3

Type RM Length L Ch R = 1 ,11697   ,14.2,13.5,13.7
XS GIS Cut Line= 3
2414498.70904024666307.5604390462414827.36936046665818.264103375
2414981.73623698665707.838105387
#Sta/Elev= 30
       0 2269.42    43.1 2245.47    63.9 2231.42      87 2214.08     102 2200.67
   126.1 2184.23   141.7 2175.91   165.1 2158.77   188.7 2139.07   205.2 2127.94
   236.9 2100.78   251.1 2092.02   270.6 2084.54   318.8 2082.51   381.5 2083.07
   391.1 2079.54   395.4 2076.89     409 2076.19   423.3 2077.35   427.1 2079.09
   437.7 2083.68     479 2083.51   502.1 2086.83     526 2093.08   545.3 2101.66
   554.9 2103.21   591.4 2105.36   677.4 2101.95   767.1 2111.13   779.2  2116.9
#Mann= 6 ,-1 , 0
       0      .1       0   288.2     .06       0   391.1    .045       0
   427.1     .06       0  433.56      .1       0  578.91     .05       0
#XS Ineff= 2 , 0
          380.54 2082.14   435.8          2081.5
Permanent Ineff=
       F       F
Bank Sta=391.1,427.1
XS Rating Curve= 0 ,0
Exp/Cntr(USF)=0,0
Exp/Cntr=0.5,0.3

Type RM Length L Ch R = 1 ,11683   ,59.1,59.3,59.8
XS GIS Cut Line= 4
2414511.04116681666316.3457269542414738.28040912665975.021834298
2414822.39508554665847.6191785282414967.70121577665729.819947922
#Sta/Elev= 30
       0 2270.09      45 2243.03    64.2  2229.5    98.9 2201.47   126.7 2182.72
   141.1  2175.2   176.8 2146.09   213.2 2118.94   237.4  2098.9   251.6 2090.04
   261.2 2085.96   269.1  2084.2   353.1  2081.2   376.6 2082.42     382 2081.63
   387.4 2078.57     391 2076.88   395.8 2076.48   400.6 2077.61   410.5 2075.91
   424.6 2078.94   434.2 2082.97   477.3  2083.5   505.8 2086.35     530 2091.67
   549.2 2100.57   562.7 2102.88   620.4 2103.23     663 2100.54   749.8 2109.04
#Mann= 5 ,-1 , 0
       0      .1       0  273.65     .06       0   387.4    .045       0
   424.6      .1       0  565.51     .05       0
Bank Sta=387.4,424.6
XS Rating Curve= 0 ,0
Exp/Cntr=0.5,0.3

Type RM Length L Ch R = 1 ,11624   ,264.9,261.1,256.9
XS GIS Cut Line= 2
2414552.13164571666347.194953462 2414986.6672572665721.411632724
#Sta/Elev= 30
       0 2271.91      28 2254.19    94.1 2202.43   125.7 2183.85   146.5 2168.96
   194.7 2130.19   204.9 2116.97   243.5 2091.25   272.3 2081.72     324 2081.93
   346.1  2078.2   370.5 2079.73   376.3 2079.08   384.3 2074.44     393 2072.47
   407.3 2072.04   419.2 2072.75     424 2074.83   438.7 2081.02   474.5 2081.26
   490.7  2083.8   550.7 2086.41   565.3 2090.96   579.9 2097.48   586.7 2098.85
   602.8 2099.68   657.8 2098.59   737.9 2107.35   749.4 2106.96   761.9 2113.49
#Mann= 5 ,-1 , 0
       0      .1       0  279.82     .06       0   384.3    .045       0
     424      .1       0  549.23     .05       0
Bank Sta=384.3,424
XS Rating Curve= 0 ,0
Exp/Cntr(USF)=0,0
Exp/Cntr=0.3,0.1

Type RM Length L Ch R = 1 ,11363   ,310.9,300,289.8
XS GIS Cut Line= 3
2414832.02499805666525.622719886     2415001.071      666156.666
     2415150.029      665754.836
#Sta/Elev= 30
       0 2286.84    64.6 2254.89   121.8 2216.68   152.6 2200.42   191.2 2175.34
     223 2153.83   240.6 2139.95   258.2  2123.9   275.8 2110.05     289 2094.33
   304.2 2084.47   324.2 2074.01   345.1 2072.33   363.2 2065.66   384.3 2064.92
   402.4  2062.2   416.3 2062.77   422.2  2065.1   436.5 2067.95   486.3 2070.81
   544.2 2067.77     557 2071.61   574.1 2071.57     604 2076.46   629.5 2084.68
     668 2086.83   723.4 2093.95   750.9 2103.48   783.1 2122.94   834.4 2150.07
#Mann= 9 ,-1 , 0
       0      .1       0  271.85     .06       0   384.3    .045       0
   422.2      .1       0  501.21     .05       0  556.18      .1       0
  612.92     .05       0  724.62      .1       0  757.57      .1       0
#XS Ineff= 2 , 0
                          485.64          2075.3
Permanent Ineff=
       F       F
Bank Sta=384.3,422.2
XS Rating Curve= 0 ,0
Exp/Cntr=0.3,0.1

Type RM Length L Ch R = 1 ,11063   ,431.5,450,468
XS GIS Cut Line= 3
     2415351.834      666589.604     2415276.805       666176.02
 2415200.4548842665773.924033774
#Sta/Elev= 30
       0 2108.64    31.2 2117.32    72.1 2119.05   120.7 2129.38   144.4 2130.24
   158.1 2126.87   173.5 2118.92     202 2096.29   222.3 2085.68   238.5 2067.33
   250.7  2063.1   283.3 2059.16   352.4 2058.13   372.7 2054.22   401.2 2054.05
   429.2 2051.07   437.8 2053.58   445.9 2058.69   454.3 2059.79     507 2061.69
     564 2058.85   580.3    2065   608.8 2080.97   661.7 2085.12   690.2  2089.9
   722.8 2103.99   775.7 2133.53   796.1 2142.68   812.3 2146.44   829.6 2154.75
#Mann= 7 ,-1 , 0
       0      .1       0  272.41     .06       0  369.98      .1       0
   401.2    .045       0   437.8      .1       0  467.56     .05       0
  662.74      .1       0
Bank Sta=401.2,437.8
XS Rating Curve= 0 ,0
Exp/Cntr=0.3,0.1

Type RM Length L Ch R = 1 ,10613   ,450.2,450,448.6
XS GIS Cut Line= 3
2415389.44274135666544.579960506     2415702.598      666238.945
2416011.80687817665970.846073585
#Sta/Elev= 30
       0 2100.13    24.2  2095.6    85.7 2093.77   102.4 2091.51   111.2 2088.39
   143.5 2065.46     157 2058.53   188.8 2051.92   242.9 2046.09   275.7 2047.21
   317.4 2042.13   409.8 2040.64   414.8  2039.9     421 2036.55   426.6 2033.86
   432.1 2033.32   449.1 2033.66   457.6 2036.29   468.2 2045.05   480.1 2060.01
   483.1 2062.17   511.5 2072.77   541.5 2089.57   564.8 2105.82   573.8 2115.87
   580.7 2120.88   627.7 2148.35   760.7 2222.78   803.5 2241.89   846.8 2258.71
#Mann= 5 ,-1 , 0
       0      .1       0   234.5     .05       0  304.87     .06       0
     421    .045       0   457.6      .1       0
Bank Sta=421,457.6
XS Rating Curve= 0 ,0
Exp/Cntr=0.3,0.1

Type RM Length L Ch R = 1 ,10163   ,201,203.9,207
XS GIS Cut Line= 3
     2415724.407       666852.36     2416013.938      666562.771
      2416303.47      666273.182
#Sta/Elev= 30
       0 2143.66    59.9 2134.77   120.9 2120.35   135.6 2110.84   150.4 2107.39
   209.2 2078.32     251 2047.11   267.9 2027.75   273.6 2024.91   308.8 2022.31
   375.4 2025.35   387.4 2024.61   392.4 2022.24   398.7 2019.64   415.6 2019.25
   427.6 2021.57   437.6 2032.08   443.9 2035.05     475 2041.19   534.4 2048.16
   545.8 2051.28   557.7  2056.3   588.2 2075.91   636.9 2102.43   669.5 2117.12
   710.5 2128.91   743.7 2146.09   761.4 2152.84     801 2160.57     819 2166.58
#Mann= 6 ,-1 , 0
       0     .05       0  205.51      .1       0  327.96     .06       0
   392.4    .045       0   427.6     .06       0   450.4      .1       0
#XS Ineff= 2 , 0
          373.72  2034.8
Permanent Ineff=
       F       F
Bank Sta=392.4,427.6
XS Rating Curve= 0 ,0
Exp/Cntr=0.3,0.1

Type RM Length L Ch R = 1 ,9959    ,57.8,57.6,58.9
XS GIS Cut Line= 3
2415804.16004287666970.6328071192416132.98604287666726.480807119
2416465.40004287666487.351807119
#Sta/Elev= 30
       0 2114.17    18.2 2112.75    33.1 2109.75     136 2078.85   192.5 2066.38
   230.4 2055.15     239 2051.36   276.1 2027.62   294.8 2019.23   307.6 2016.62
   402.2 2016.89   408.9  2015.4   416.3 2012.01   427.7 2011.79   441.3 2012.93
   447.8 2015.63   456.1 2017.82   482.2 2017.09   502.2 2018.75   511.6 2022.33
     530 2035.38   536.6 2038.09   569.4 2040.01   586.9 2042.96   607.5 2058.19
   702.4 2122.28   727.1 2135.04   765.9 2161.63   781.3 2173.79     819 2196.02
#Mann= 5 ,-1 , 0
       0      .1       0  344.08     .06       0   408.9    .045       0
   447.8     .06       0  455.58      .1       0
#XS Ineff= 2 , 0
          392.58 2021.14
Permanent Ineff=
       F       F
Bank Sta=408.9,447.8
XS Rating Curve= 0 ,0
Exp/Cntr=0.5,0.3

Type RM Length L Ch R = 1 ,9901    ,28.8,29.3,30.2
XS GIS Cut Line= 3
 2415828.5929645666979.5858244262416225.88080785666735.100997746
2416490.38809879666524.338216125
#Sta/Elev= 30
       0 2102.02      26 2096.44   100.9 2068.18   148.1 2061.01   182.3 2052.38
   192.1 2047.91   214.3 2045.56   218.6 2043.47   228.9 2032.22     255 2021.99
   283.7 2015.57   306.6  2016.5   397.5 2016.16   405.3 2012.27   411.1 2009.83
   420.5 2009.36   432.4 2011.94   441.1  2015.9   509.9 2015.49   518.2 2019.01
   537.4 2033.11   569.5 2038.77   601.6 2052.37   640.1 2076.43   672.2 2100.95
   717.2 2131.55   736.4 2147.26   757.6 2159.04   781.3 2175.82   804.7 2189.82
#Mann= 4 ,-1 , 0
       0      .1       0   306.6     .06       0   405.3    .045       0
   432.4      .1       0
#XS Ineff= 3 ,-1
       0     386    2018     386   398.2    2014     444     560    2014
Permanent Ineff=
       F       F       F
Bank Sta=405.3,432.4
XS Rating Curve= 0 ,0
Exp/Cntr(USF)=0,0
Exp/Cntr=0.5,0.3

Type RM Length L Ch R = 1 ,9872    ,58.2,56.9,53.8
XS GIS Cut Line= 4
2415836.45207339 666997.589073392416002.81804852666899.133731863
 2416227.0274956 666769.008790492416522.23862365666532.417218751
#Sta/Elev= 30
       0 2092.84    16.6 2089.03    58.4  2072.5    72.4 2068.33   137.5 2067.11
   216.4 2052.72   234.9 2045.68   244.1 2037.49   267.2 2027.12   285.7 2016.47
   301.7 2014.53   401.2  2014.4   412.9 2010.69   419.8 2008.36   429.1 2008.29
     443 2011.34     451 2013.94   510.8 2013.81     524 2019.83   542.1 2031.93
   559.8 2033.03   573.4  2035.8   593.3 2042.48   609.4 2051.48   621.7 2055.63
   630.3 2060.63   698.2 2110.41   764.9 2153.44   794.9 2177.45   830.9 2198.75
#Mann= 5 ,-1 , 0
       0      .1       0  298.22     .06       0   412.9    .045       0
     443     .06       0  449.17      .1       0
#XS Ineff= 2 , 0
          393.22 2023.79
Permanent Ineff=
       F       F
Bank Sta=412.9,443
XS Rating Curve= 0 ,0
Exp/Cntr=0.5,0.3

Type RM Length L Ch R = 1 ,9815    ,256.5,252.4,247.8
XS GIS Cut Line= 3
2415919.12689625667079.2287190732416239.90889625666825.659719073
2416557.87089625666562.235719073
#Sta/Elev= 30
       0 2099.86    71.5 2095.41   121.9 2089.78   194.1 2077.32   213.7 2069.78
   234.1 2059.27   239.2 2054.83   247.7 2043.04   256.3 2035.65   269.7 2026.63
   290.1 2015.36   303.7 2013.26   366.6 2011.95   387.3  2009.9   397.2 2006.88
   402.3 2005.84     432 2006.99   485.3    2012   511.3 2028.43   516.5 2030.41
   557.8 2032.31     572 2034.92   588.8 2041.91     610 2056.18   626.4 2063.83
   694.1 2114.46   720.5 2129.65   750.9 2153.42   786.6 2177.22   821.8 2197.95
#Mann= 5 ,-1 , 0
       0      .1       0  326.01     .06       0   397.2    .045       0
     432     .06       0  467.84      .1       0
Bank Sta=397.2,432
XS Rating Curve= 0 ,0
Exp/Cntr=0.3,0.1

Type RM Length L Ch R = 1 ,9563    ,452.8,450,446.9
XS GIS Cut Line= 3
     2416172.645      667348.736     2416404.575      667011.332
     2416644.635      666679.083
#Sta/Elev= 30
       0 2172.14      32 2162.82    79.9 2144.34   104.2  2132.9   144.9 2110.98
   152.7 2108.45   207.1 2080.96   247.3 2057.76   258.9 2055.69   303.2 2024.45
     342 2003.14   385.7 2002.62     394 1999.04     410 1995.71     420 1996.47
   425.6 1999.31   445.7 2004.19   503.7 2002.05   518.5 2003.67   538.3 2002.89
   548.2 2006.08   567.9 2020.42   604.4 2024.56   617.6 2030.93   666.3 2060.31
     711 2091.24   726.4 2105.12   745.5 2119.58     790 2147.22   819.3 2169.04
#Mann= 5 ,-1 , 0
       0      .1       0  290.77     .06       0     394    .045       0
   425.6     .06       0  433.89      .1       0
#XS Ineff= 2 , 0
                          448.96         2008.66
Permanent Ineff=
       F       F
Bank Sta=394,425.6
XS Rating Curve= 0 ,0
Exp/Cntr=0.3,0.1

Type RM Length L Ch R = 1 ,9113    ,545.1,546.9,551.5
XS GIS Cut Line= 3
      2416654.76       667554.94     2416820.516      667169.583
     2416980.061      666794.357
#Sta/Elev= 30
       0 2109.64    60.9 2083.45   152.9 2038.57   172.1 2031.78   187.3 2023.15
   225.3 2005.35   255.8 1992.48   274.4 1992.51   283.2  1991.3   295.4 1984.37
   300.5 1983.47   335.3 1988.15   370.2 1986.57   383.7 1989.23   391.9 1987.69
     405 1982.01   411.1 1980.19   425.2 1979.63   444.2 1980.71   448.5 1982.23
   461.5 1990.63   470.2 1993.32   487.6 1995.02     492 1997.02     518 2013.76
   570.2 2039.64   697.7 2112.36   744.1 2134.61   795.3 2160.77   827.2 2174.49
#Mann= 5 ,-1 , 0
       0      .1       0  186.88     .06       0  302.03      .1       0
     405    .045       0   448.5      .1       0
#XS Ineff= 2 , 0
          387.06 2003.07
Permanent Ineff=
       F       F
Bank Sta=405,448.5
XS Rating Curve= 0 ,0
Exp/Cntr=0.3,0.1

Type RM Length L Ch R = 1 ,8566    ,88.4,88.3,88.7
XS GIS Cut Line= 3
2417072.21551223667835.4827914552417266.44451223667475.428791455
2417455.39251223667109.914791455
#Sta/Elev= 30
       0 2132.84   105.2 2077.28   155.8 2046.11     187 2029.17     216 2009.91
   259.7 1975.51   279.8 1969.02   296.1 1966.26   389.1 1967.53     392 1967.28
   397.9 1964.21   403.8 1961.27   412.7 1960.61   418.7 1961.19   424.6 1964.26
   432.2 1968.07   439.4 1969.41   450.2 1966.82   468.2 1967.36   486.3 1977.75
   498.8 1986.38   531.4 2013.79   656.1 2099.86   670.9 2111.83   688.8 2123.01
   702.4 2135.48   733.9 2158.58   748.1 2168.05   792.4 2193.28   820.6 2210.81
#Mann= 5 ,-1 , 0
       0      .1       0  304.17     .06       0   397.9    .045       0
   424.6     .06       0  468.49      .1       0
#XS Ineff= 2 , 0
          386.14 1972.98  439.36         1974.75
Permanent Ineff=
       F       F
Bank Sta=397.9,424.6
XS Rating Curve= 0 ,0
Exp/Cntr=0.5,0.3

Type RM Length L Ch R = 1 ,8478    ,37.9,37.4,37.3
XS GIS Cut Line= 2
2417139.79164695667864.3030813782417564.82992322667139.513293467
#Sta/Elev= 30
       0 2131.07    38.3 2110.24   128.9 2057.47   187.1 2017.44   219.6 1996.92
   247.4 1974.66   261.3 1967.46     275 1963.62   359.8 1963.29   394.9 1965.02
   397.8 1963.98   403.6  1959.2   409.1 1956.24   414.3 1955.34     419 1956.35
   423.6 1959.52   428.2 1963.82   432.9 1965.53   470.9 1962.34   493.2 1963.78
   497.8 1967.22   511.7  1983.4   539.5 2006.45   559.3 2020.31   637.5 2071.53
     674 2098.06   734.3  2135.7   769.3  2162.9   803.8 2183.05   840.2  2201.1
#Mann= 5 ,-1 , 0
       0      .1       0  317.36     .06       0   403.6    .045       0
   423.6     .06       0  443.26      .1       0
#XS Ineff= 2 , 0
          385.06 1971.94  434.92         1972.39
Permanent Ineff=
       F       F
Bank Sta=403.6,423.6
XS Rating Curve= 0 ,0
Exp/Cntr(USF)=0,0
Exp/Cntr=0.5,0.3

Type RM Length L Ch R = 1 ,8440    ,70.1,70.3,70
XS GIS Cut Line= 2
2417172.57696853667878.353933486 2417597.6152448667158.247762945
#Sta/Elev= 30
       0 2130.42    50.5 2101.79    91.7 2074.73     118 2060.23     148  2036.1
   208.6 1996.44   236.3 1972.97   240.9 1970.56   268.8 1965.93   278.1 1961.17
   305.9 1962.77   375.1 1963.26   383.8 1962.09   389.9 1958.35   394.2  1955.3
   398.8  1954.4   405.6 1955.21   412.8 1958.59   424.7 1964.61   473.1 1960.61
     486  1961.7   496.4 1965.46   556.1 2013.61   617.1 2054.77   655.5 2078.48
   714.7 2119.51   740.2 2134.38   761.1 2151.66   802.9 2175.56   836.2 2191.05
#Mann= 5 ,-1 , 0
       0      .1       0  300.99     .06       0   389.9    .045       0
   412.8     .06       0  456.27      .1       0
#XS Ineff= 2 , 0
          372.55 1966.96  426.36          1967.5
Permanent Ineff=
       F       F
Bank Sta=389.9,412.8
XS Rating Curve= 0 ,0
Exp/Cntr(USF)=0,0
Exp/Cntr=0.5,0.3

Type RM Length L Ch R = 1 ,8370    ,469,457.1,444.9
XS GIS Cut Line= 3
2417213.50868156667900.9455947152417416.42057145667596.628206498
2417673.08584561667221.582782883
#Sta/Elev= 30
       0 2133.66    51.4 2104.35    62.9 2094.79     113 2060.83   139.2 2039.76
     190 2002.48   218.8 1976.82   228.4 1970.21   247.5  1965.2   276.5  1962.9
   287.9 1959.75   358.2 1961.09   362.9 1960.92   368.7 1958.44     377 1953.81
   383.1 1953.11   401.8 1958.35     409 1960.22   445.4 1958.47   469.4 1959.47
     523 1974.51   595.7  2018.6   605.4 2024.98   615.1 2034.98   653.6 2056.62
   678.1 2072.94   699.6  2085.3   752.3 2111.42   794.4 2128.99   820.2 2136.32
#Mann= 4 ,-1 , 0
       0      .1       0  265.76     .06       0   368.7    .045       0
   401.8      .1       0
#XS Ineff= 2 , 0
          355.92 1964.09  411.98         1964.48
Permanent Ineff=
       F       F
Bank Sta=368.7,401.8
XS Rating Curve= 0 ,0
Exp/Cntr=0.3,0.1

Type RM Length L Ch R = 1 ,7913    ,340.6,354.6,367.7
XS GIS Cut Line= 4
2417753.44735345668114.2657901082417842.93445627667889.198448656
     2417834.258      667696.308     2417808.484      667288.675
#Sta/Elev= 30
       0 2038.92    42.4 2022.76    55.3 2015.24    76.8 2006.08      94 2003.09
   145.7 1981.12   175.8  1975.4   201.6 1973.98   223.2 1976.53   264.5 1988.12
   308.6 1985.37   320.6 1981.85   340.9 1972.11   344.6 1969.83   352.6 1959.64
   368.6 1948.87   392.7 1949.23     4081940.383   416.7 1938.12   440.7 1937.44
   451.2 1940.23   460.8 1945.93   512.9 1946.47   532.9 1959.49     565 1969.11
   591.4 1981.33   641.1 2010.93   693.2  2025.5   753.3 2060.19   843.7 2095.88
#Mann= 4 ,-1 , 0
       0      .1       0  328.54     .06       0     408    .045       0
   451.2      .1       0
Bank Sta=408,451.2
XS Rating Curve= 0 ,0
Exp/Cntr=0.3,0.1

Type RM Length L Ch R = 1 ,7558    ,72.3,74.4,75.3
XS GIS Cut Line= 2
2417847.56667592 668050.929410172418476.34230776667543.927829934
#Sta/Elev= 30
       0 2034.76    12.8 2029.42    25.6 2027.27    31.9 2023.46    38.3 2022.89
    56.3 2016.07    70.2 2012.93    82.9 2012.59   121.1 2016.63   212.8 2009.09
     255 2002.57   274.1 2004.58   295.3 1995.31     301 1990.43   306.7 1979.13
   318.7    1949   325.1 1940.55   331.4 1935.11   356.9 1933.45   380.6 1925.54
   394.11926.272   404.9 1924.06   415.2 1926.99   425.4 1931.62   507.6 1932.73
   522.6 1936.53   551.3 1963.23   567.2 1975.56   669.2 2042.27   807.7 2139.15
#Mann= 4 ,-1 , 0
       0      .1       0  286.63     .06       0   394.1    .045       0
   415.2      .1       0
Bank Sta=394.1,415.2
XS Rating Curve= 0 ,0
Exp/Cntr(USF)=0,0
Exp/Cntr=0.5,0.3

Type RM Length L Ch R = 1 ,7484    ,28.8,29.5,33.4
XS GIS Cut Line= 2
2417867.05189778668089.5636860772418556.38498097 667612.49264555
#Sta/Elev= 30
       0 2061.62    92.1 2050.62   166.4 2030.45   187.4 2021.53   263.3 2018.39
   296.4 2002.85   315.1  1984.1   320.7 1975.82   330.4 1951.69   335.2    1942
   340.1    1938   356.1 1931.66   386.9 1930.47   398.4 1925.47   408.2 1923.84
   427.2 1922.37   437.4  1924.1     452 1928.82     525 1929.75   534.7 1931.84
     560 1947.34   582.4 1964.41   605.4 1978.06   616.2 1990.38   622.3 1995.08
   657.2 2013.37   743.9 2072.96   784.9 2104.99   802.3  2116.3   838.3  2145.6
#Mann= 4 ,-1 , 0
       0      .1       0  261.42     .06       0   408.2    .045       0
   437.4      .1       0
#XS Ineff= 2 , 0
           408.2    1923   437.4            1923
Permanent Ineff=
       F       F
Bank Sta=408.2,437.4
XS Rating Curve= 0 ,0
Exp/Cntr(USF)=0,0
Exp/Cntr=0.5,0.3

Type RM Length L Ch R = 1 ,7454    ,63.6,63.9,64.6
XS GIS Cut Line= 3
2417884.43060005668110.5658913482418111.05721806667951.650975618
2418582.00720867667642.358939653
#Sta/Elev= 30
       0  2075.1    87.6 2060.78   139.6 2049.38   173.6 2037.69   188.5 2035.52
   208.4 2025.89   229.3 2023.41   262.8 2023.16   288.7 2009.01   295.6 2004.82
   300.2 2000.53     306 1990.81   314.7 1980.01   329.1 1948.43   333.8 1944.17
   348.2 1935.67   358.3 1931.55   386.9 1929.98   407.1 1923.76   430.2 1921.82
   443.9 1922.02   450.4 1923.93     462 1926.58   506.1 1928.03   534.2  1931.3
     554 1939.72   574.6 1954.11   632.4 1990.37   692.8 2031.56   840.2 2138.28
#Mann= 5 ,-1 , 0
       0      .1       0  262.36     .06       0   407.1    .045       0
   450.4     .06       0  464.87      .1       0
Bank Sta=407.1,450.4
XS Rating Curve= 0 ,0
Exp/Cntr=0.5,0.3

Type RM Length L Ch R = 1 ,7390    ,47.2,47.4,47.6
XS GIS Cut Line= 2
2417917.95103694668146.0328628652418620.49364235667702.260117116
#Sta/Elev= 30
       0 2094.02    34.1 2088.51   101.4 2071.29   133.8 2065.57   178.2 2050.89
   194.9 2048.27   230.6 2037.46   261.2 2022.62   284.8 2005.49   301.5 1981.69
   313.2 1953.58   317.9  1947.9   324.7 1942.97   336.3 1935.39     351 1930.23
   385.6 1928.03   400.1 1922.26     422 1918.38   434.9 1922.67   445.7 1926.25
   455.2 1924.75   516.1 1925.96   537.7 1930.69   571.2 1953.32   614.7 1974.33
   652.4 1997.25   696.4 2027.86   739.4 2055.38   782.8 2089.63     831 2124.49
#Mann= 4 ,-1 , 0
       0      .1       0  319.68     .06       0   400.1    .045       0
   434.9      .1       0
Bank Sta=400.1,434.9
XS Rating Curve= 0 ,0
Exp/Cntr(USF)=0,0
Exp/Cntr=0.5,0.3

Type RM Length L Ch R = 1 ,7343    ,16.4,16.6,16.8
XS GIS Cut Line= 2
2417948.15059286668175.3595638042418645.19190367667749.495968436
#Sta/Elev= 30
       0 2110.87   148.4 2072.01   199.9 2054.93   218.7 2040.63   237.9 2023.44
   261.8 2006.38   265.5 2002.58   272.8 1989.47   284.3 1978.44   298.4 1959.71
   328.1 1936.37   336.8 1930.62   345.2 1927.81   374.7 1926.05   387.4 1921.61
   396.8 1917.84   406.2 1917.04   418.3 1918.45   424.9 1921.41   432.9 1923.56
   502.7 1924.15     514 1925.75   551.5 1946.35   593.7 1963.45     622  1979.6
   682.7 2020.16   771.8 2084.49   779.1  2091.4   808.2 2110.27   816.8 2119.76
#Mann= 4 ,-1 , 0
       0      .1       0   328.1     .06       0   387.4    .045       0
   424.9      .1       0
#XS Ineff= 2 , 0
          376.99 1925.99     436         1926.13
Permanent Ineff=
       F       F
Bank Sta=387.4,424.9
XS Rating Curve= 0 ,0
Exp/Cntr(USF)=0,0
Exp/Cntr=0.5,0.3

Type RM Length L Ch R = 1 ,7326    ,26.9,27.7,28.3
XS GIS Cut Line= 2
2417950.06029509668187.4543445392418647.10160589667773.685529907
#Sta/Elev= 30
       0 2115.55     159  2074.1   200.8 2059.52   210.1 2052.59   224.1 2036.29
   261.3 2008.59   265.9 2003.63   270.6 1994.53   275.2 1987.78     284 1978.18
   304.5 1958.12   326.4 1941.38   339.5 1932.18   349.7 1926.95   382.2 1924.84
     392 1920.07   400.8 1917.22   414.8 1917.01   424.1 1920.28   433.4 1923.11
   507.8  1923.7   526.3 1929.33   554.3 1943.64   586.9  1956.8   640.2 1987.98
   684.6 2017.96   721.8 2045.52   769.1  2076.3   784.7 2089.72   810.6 2107.11
#Mann= 4 ,-1 , 0
       0      .1       0   326.4     .06       0     392    .045       0
   424.1      .1       0
#XS Ineff= 2 , 0
                          444.83         1925.77
Permanent Ineff=
       F       F
Bank Sta=392,424.1
XS Rating Curve= 0 ,0
Exp/Cntr(USF)=0,0
Exp/Cntr=0.5,0.3

Type RM Length L Ch R = 1 ,7299    ,140,142.5,144.9
XS GIS Cut Line= 2
2417955.78940175668197.6394230532418677.65684143667806.787035077
#Sta/Elev= 30
       0 2119.94     137 2084.09   171.7 2073.66     199 2063.04   208.1 2056.23
   217.1 2038.61   263.9 2001.68   267.2 1998.02   280.8 1976.64   317.9 1944.26
   335.4 1932.76   353.6 1925.04   358.2 1923.73   377.5 1924.23   387.4 1920.89
   394.5 1916.87   403.6 1916.04   417.3 1916.65   426.2 1920.98     435 1923.71
     481 1921.92   512.8 1924.66   526.3 1928.96   549.2 1940.57   588.5 1957.04
   617.4 1973.05   682.9 2015.76   730.1 2049.13   753.5 2064.02   820.9 2112.84
#Mann= 4 ,-1 , 0
       0      .1       0   377.5     .06       0   387.4    .045       0
   426.2      .1       0
Bank Sta=387.4,426.2
XS Rating Curve= 0 ,0
Exp/Cntr(USF)=0,0
Exp/Cntr=0.3,0.1

Type RM Length L Ch R = 1 ,7156    ,257.5,259.3,261.4
XS GIS Cut Line= 2
 2417956.3406332668294.3330361862418786.73507078667973.097276968
#Sta/Elev= 30
       0 2147.97    71.2 2135.31   152.1 2110.33   196.3 2089.77   234.2 2068.73
   238.5 2064.47   242.4  2057.8     247 2046.48   251.9 2037.41   294.2 2003.32
   319.9 1977.39   353.2  1950.6   397.2 1922.84   418.9 1922.04   431.3 1915.55
     440 1912.82   452.8 1912.47   470.1 1915.32   487.2 1918.24   547.3 1919.14
   571.8 1930.21   581.6 1937.38   632.3 1962.65   706.5 2009.05   737.5 2026.03
   749.8 2034.92   759.1  2044.1   791.7 2064.67   804.6 2074.67   890.4 2128.52
#Mann= 5 ,-1 , 0
       0      .1       0  387.65     .06       0   431.3    .045       0
   470.1     .06       0  489.16      .1       0
Bank Sta=431.3,470.1
XS Rating Curve= 0 ,0
Exp/Cntr(USF)=0,0
Exp/Cntr=0.3,0.1

Type RM Length L Ch R = 1 ,6897    ,55.9,57.1,59
XS GIS Cut Line= 3
2418059.95475554668487.3783207212418455.22775554668376.134320721
2418858.39176519668267.287229049
#Sta/Elev= 30
       0  2115.5      74 2091.02   169.1 2054.33   248.1 2014.35   277.2 1996.48
   289.6 1982.27   302.1 1972.28   314.6  1953.6   331.2 1939.17   347.8 1927.94
   360.3 1915.85   364.4 1913.97   393.5 1911.85   400.5 1907.61     406 1904.98
   414.3 1904.81   440.6 1907.51   447.4 1909.11   504.7 1910.47   530.3 1918.75
   559.3 1941.59   592.4 1963.48   600.7 1971.49   625.6 1985.67   646.6 2000.36
   650.4 2003.51   658.7 2014.47   770.6 2073.95   791.3 2086.54   828.2 2113.24
#Mann= 4 ,-1 , 0
       0      .1       0  309.88     .06       0   400.5    .045       0
   440.6      .1       0
Bank Sta=400.5,440.6
XS Rating Curve= 0 ,0
Exp/Cntr=0.5,0.3

Type RM Length L Ch R = 1 ,6840    ,17.9,17.7,18
XS GIS Cut Line= 2
 2418067.1523154668508.081664268 2418863.3672682668355.864099762
#Sta/Elev= 30
       0 2109.31   105.5 2071.56   150.3 2052.15   195.5 2027.79   235.8 2012.82
   264.3 2000.17   276.5 1991.72   280.6    1985   291.3 1962.27   300.9 1946.45
   305.1 1941.61   353.9 1911.52   390.4 1909.01   398.7 1905.65   410.9 1902.78
   427.2 1903.38   434.9 1905.82   443.5 1907.31   488.3 1907.59   504.6 1911.74
   520.3 1923.54   533.1 1927.34   553.4  1944.3     586 1964.22   602.3 1977.33
   637.4 2001.35   687.8 2031.03   781.5 2080.03   801.9    2093   810.6 2102.21
#Mann= 4 ,-1 , 0
       0      .1       0  304.21     .06       0   398.7    .045       0
   434.9      .1       0
#XS Ineff= 2 , 0
           398.7    1904   434.9            1904
Permanent Ineff=
       F       F
Bank Sta=398.7,434.9
XS Rating Curve= 0 ,0
Exp/Cntr(USF)=0,0
Exp/Cntr=0.5,0.3

Type RM Length L Ch R = 1 ,6822    ,49.6,50.3,52.1
XS GIS Cut Line= 2
2418068.44716485668520.9414566232418871.17104608 668377.12873716
#Sta/Elev= 30
       0 2106.76    95.8 2071.86   156.8 2044.81   193.3 2024.76   254.3 2001.87
   262.4 1997.41   266.5 1992.53   270.5 1984.77   278.7 1974.76   294.9 1948.92
     299 1943.01     303 1939.86   351.8 1910.65   393.2 1908.77   403.5 1904.69
   408.7 1902.69   416.8  1902.5     429 1902.81   437.1 1904.84   445.3 1906.45
   485.9 1906.51   498.1 1910.31   526.6 1929.57   538.7 1933.41   611.9 1984.55
   658.7  2013.3   733.8  2054.3   787.5 2080.68   807.3 2093.26   815.5 2100.42
#Mann= 4 ,-1 , 0
       0      .1       0  304.91     .06       0   403.5    .045       0
   437.1      .1       0
Bank Sta=403.5,437.1
XS Rating Curve= 0 ,0
Exp/Cntr(USF)=0,0
Exp/Cntr=0.5,0.3

Type RM Length L Ch R = 1 ,6772    ,203.2,208.9,212.5
XS GIS Cut Line= 2
2418073.73045917668549.7053137152418869.46534118668447.274601846
#Sta/Elev= 30
       0 2099.76    81.7 2069.14    97.8 2061.92   138.1 2041.04     247 1991.14
   263.2 1979.89   267.2 1973.82   283.3 1941.78   287.4 1938.03   328.6 1913.76
   343.8 1907.47   400.3 1907.31   404.3 1906.94   408.4 1904.73   412.4 1902.16
   416.4 1901.43   436.6 1901.49   446.9 1904.51   497.1 1906.19   501.1 1908.35
   509.2 1918.45   529.3 1935.61   533.4 1938.21     543 1941.23   565.6 1957.65
   626.1 1998.36   639.4 2006.34   692.2  2033.7   722.9 2047.73   802.3 2079.01
#Mann= 5 ,-1 , 0
       0      .1       0  304.42     .06       0   408.4    .045       0
   446.9     .06       0  503.16      .1       0
Bank Sta=408.4,446.9
XS Rating Curve= 0 ,0
Exp/Cntr(USF)=0,0
Exp/Cntr=0.3,0.1
